--- 2ndBroadRv.prj (project) ---

Proj Title=2ndBroadRv
Current Plan=p01
Default Exp/Contr=0.3,0.1
English Units
Geom File=g01
Flow File=f01
Plan File=p01
Y Axis Title=Elevation
X Axis Title(PF)=Main Channel Distance
X Axis Title(XS)=Station
BEGIN DESCRIPTION:
END DESCRIPTION:
DSS Export Rating Curves= 0
DSS Export Rating Curve Sorted= 0
DSS Export Volume Flow Curves= 0
DXF OffsetX= 0
DXF OffsetY= 0
DXF ScaleX= 1
DXF ScaleY= 10

--- 2ndBroadRv.p01 (plan) ---

Plan Title=LD Study - 100 YR
Program Version=3.12
Short Identifier=lds
Geom File=g01
Flow File=f01
Subcritical Flow
K Sum by GR= 0
Std Step Tol= 0.01
Critical Tol= 0.01
Num of Std Step Trials= 20
Max Error Tol= 0.3
Flow Tol Ratio= 0.001
Split Flow NTrial= 30
Split Flow Tol= 0.02
Split Flow Ratio= 0.02
Log Output Level= 0
Friction Slope Method= 1
Unsteady Friction Slope Method= 2
Unsteady Bridges Friction Slope Method= 1
Calc Critical at every XS
Parabolic Critical Depth
Global Vel Dist= 0 , 0 , 0
Global Log Level= 0
CheckData=True
Encroach Param=-1 ,10,10, 2
Encroach River=2ndBroadRv
Encroach Reach=Main
Encroach Node=241211.7
       1  500.97     545
Encroach Node=240211.7
       1  456.21  525.72
Encroach Node=239342.5
       1     875  981.45
Encroach Node=238211.7
       1  834.83     950
Encroach Node=237299.1
       1  207.04  259.23
Encroach Node=237209.0
       1  168.09  217.08
Encroach Node=237112.9
       1  190.82  239.81
Encroach Node=236621.8
       1  356.73  533.98
Encroach Node=236044.7
       1  331.09  504.73
Encroach Node=235211.7
       1  659.27  710.15
Encroach Node=234211.7
       1  682.34   738.8
Encroach Node=233027.8
       1  740.02  829.74
Encroach Node=232462.0
       1  417.25  460.81
Encroach Node=232353.0
       1  417.25  487.01
Encroach Node=232213.3
       1  477.33  547.09
Encroach Node=231827.0
       1  421.84  576.82
Encroach Node=231211.7
       1  624.63  775.64
Encroach Node=230211.7
       1  606.19  703.16
Encroach Node=229729.2
       1  367.45  515.21
Encroach Node=229416.7
       1  333.13  425.83
Encroach Node=229347.1
       1   352.8  445.51
Encroach Node=228874.8
       1   781.7  886.66
Encroach Node=228454.6
       1  885.55 1035.67
Encroach Node=227553.7
       1  369.05     547
Encroach Node=227418.4
       1  144.99  382.02
Encroach Node=227337.8
       1  147.11  384.13
Encroach Node=226917.6
       1   558.3  701.62
Encroach Node=225677.0
       1  782.37   837.9
Encroach Node=224964.2
       1  375.96  688.08
Encroach Node=224772.5
       1  616.23  860.62
Encroach Node=224606.8
       1  281.62  412.44
Encroach Node=223974.5
       1  241.84  335.85
Encroach Node=223682.1
       1  746.69    1035
Encroach Node=223159.2
       1   86.92  163.35
Encroach Node=222727.8
       1    1111    1146
Encroach Node=222497.9
       1  456.48  525.34
Encroach Node=222391.5
       1  418.35  487.21
Encroach Node=221965.6
       1  571.67 1130.42
Encroach Node=220678.9
       1  937.06 1130.94
Encroach Node=220186.1
       1  770.29  841.21
Encroach Node=218965.2
       1   919.9  981.55
Encroach Node=217791.7
       1  325.49   446.1
Encroach Node=217686.7
       1   382.2   435.7
Encroach Node=217600.6
       1     225     280
Encroach Node=217473.4
       1     320  394.51
Encroach Node=217400.1
       1  332.13  450.76
Encroach Node=217260.7
       1   316.4   370.5
Encroach Node=216927.3
       1    78.4  128.64
Encroach Node=216521.8
       1    54.8     112
Encroach Node=216121.1
       1   55.85    94.7
Encroach Node=215827.1
       1      72     151
Encroach Node=215654.2
       1      51    95.4
Encroach Node=215376.6
       1   34.22  120.62
Encroach Node=215037.2
       1     110  187.48
Encroach Node=214740.5
       1     200     348
Encroach Node=214517.8
       1 1234.12    1292
Encroach Node=214079.0
       1     500   571.7
Encroach Node=213566.3
       1   363.9     468
Encroach Node=213365.4
       1  108.14  202.07
Encroach Node=213235.3
       1     150  241.37
Encroach Node=213153.9
       1  619.08  684.06
Encroach Node=212461.4
       1   375.7  449.09
Encroach Node=211897.6
       1     830  884.66
Encroach Node=211122.6
       1     274     330
Encroach Node=210211.7
       1  960.87 1035.37
Encroach Node=209331.1
       1     235     420
Encroach Node=208845.5
       1  849.81 1134.17
Encroach Node=208483.1
       1 1114.18 1180.54
Encroach Node=207883.3
       1   133.7     178
Encroach Node=207664.1
       1   401.4   447.4
Encroach Node=207574.0
       1  118.95  207.54
Encroach Node=207406.6
       1  156.13  244.72
Encroach Node=207086.1
       1  460.13  611.64
Encroach Node=206307.5
       1  378.45  424.48
Encroach Node=206252.2
       1  150.57  271.96
Encroach Node=206189.5
       1  151.26     260
Encroach Node=206082.3
       1  474.35  574.09
Encroach Node=205899.4
       1  550.72  685.22
Encroach Node=205545.2
       1     365  474.92
Encroach Node=204964.6
       1  212.23  276.06
Encroach Node=204556.1
       1  261.33  330.13
Encroach Node=204484.8
       1  108.09   169.1
Encroach Node=204369.3
       1    48.6   138.5
Encroach Node=204187.8
       1     440     530
Encroach Node=203618.5
       1     679     950
Encroach Node=203250.0
       1  827.12  930.83
Encroach Node=202036.8
       1  555.47   793.4
Encroach Node=201455.3
       1  597.57   763.1
Encroach Node=200576.0
       1   708.7   889.2
Encroach Node=199211.7
       1  693.51 1025.85
Encroach Node=198005.1
       1 1037.15 1339.44
Encroach Node=197211.7
       1  518.23  825.53
Encroach Node=196211.7
       1  455.86   832.5
Encroach Node=195239.8
       1  346.83  842.91
Encroach Node=193888.7
       1  443.07  535.99
Encroach Node=193211.7
       1  646.23  719.25
Encroach Node=192437.0
       1  431.77  509.32
Encroach Node=192244.8
       1     215  446.77
Encroach Node=192096.6
       1     240     517
Encroach Node=191849.6
       1  446.77  523.32
Encroach Node=190944.2
       1  572.38  804.67
Encroach Node=190221.7
       1  588.64  945.91
Encroach Node=188988.4
       1  540.47  809.64
Encroach Node=187481.
       1  675.25   756.6
Computation Interval=1HOUR
Output Interval=1HOUR
Run HTab= 0
Run UNet= 0
Run PostProcess= 0
UNET Theta= 1
UNET Theta Warmup= 1
UNET ZTol= 0.02
UNET ZSATol= 0.05
UNET MxIter= 20
UNET MaxInSteps= 0
UNET DtIC= 0
UNET DtMin= 0
UNET MaxCRTS= 20
UNET WFStab= 2
UNET SFStab= 1
UNET WFX= 1
UNET SFX= 1
UNET DSS MLevel= 4
UNET DZMax Abort= 100
UNET Convert EG Bridges=-1
UNET Use Existing IB Tables=-1
UNET Froude Reduction=False
UNET Froude Limit= 1
UNET Froude Power= 10
Instantaneous Interval=1HOUR
Write IC File= 0
Echo Input=False
Echo Output=False
Write Detailed= 0
Detailed Automatic Start=False, 10

--- 2ndBroadRv.f01 (steady flow) ---

Flow Title=2ndBroadRv
Program Version=3.12
Number of Profiles= 2
Profile Names=P100yr,Encroachments
River Rch & RM=2ndBroadRv,Main            ,241211.7
    1560    1560
River Rch & RM=2ndBroadRv,Main            ,238211.7
    1760    1760
River Rch & RM=2ndBroadRv,Main            ,236621.8
    1900    1900
River Rch & RM=2ndBroadRv,Main            ,235211.7
    2090    2090
River Rch & RM=2ndBroadRv,Main            ,228874.8
    2400    2400
River Rch & RM=2ndBroadRv,Main            ,225677.0
    3300    3330
River Rch & RM=2ndBroadRv,Main            ,220186.1
    3980    3980
River Rch & RM=2ndBroadRv,Main            ,214517.8
    4200    4200
River Rch & RM=2ndBroadRv,Main            ,208845.5
    4630    4630
River Rch & RM=2ndBroadRv,Main            ,205899.4
    5080    5080
River Rch & RM=2ndBroadRv,Main            ,198005.1
    6040    6040
Boundary for River Rch & Prof#=2ndBroadRv,Main            , 1
Up Type= 0
Dn Type= 3
Dn Slope=0.005
DSS Import GetInterval= 0
DSS Import GetPeak= 0
DSS Import FillOption= 0

--- 2ndBroadRv.g01 (geometry) ---

Geom Title=2ndBroadRv
Program Version=3.12

River Reach=2ndBroadRv      ,Main
Reach XY= 30
  1096817.378174   688665.878274  1100347.999093    685097.05806
  1101705.749341   684354.559736  1103237.002081   682448.309997
  1105014.748042   681894.502138  1106584.879987   682044.497668
  1108900.877158   679243.128566  1109275.878245   679857.692405
  1110314.128239   679758.749435  1110657.880935   679477.501696
  1110498.132851   678753.558247  1111678.628727    678284.81203
  1113480.749962   678177.189616  1113286.378368    678524.37887
  1113959.883641   679142.440706  1113942.631281   678368.128739
  1115407.881067   677397.630719  1117466.878853   672909.811464
  1118373.131158   671970.561791  1118091.875201   670843.809509
  1117154.382723   670524.378868  1117234.250612   669935.808228
  1118484.251526   669130.309352  1118959.879034   667470.561007
  1119761.998702   666833.440482  1119699.497877   665927.192309
   1118345.38072   664296.939247  1118328.001395   663340.379862
  1115734.250351   658994.880233  1115827.999612   657276.129015

Type RM Length L Ch R = 1 ,241211.7,999.84,1000,1002.03
BEGIN DESCRIPTION:
53943.71
END DESCRIPTION:
XS GIS Cut Line= 3
  1097190.777062   689031.962781  1096824.033036   688658.414183
  1096505.167113   688366.717455
#Sta/Elev= 30
       0 1399.03   38.58 1393.37   80.66 1388.73  144.02 1379.56  223.92 1372.41
  270.73 1370.76  379.05  1370.3  486.19  1367.8  500.32 1365.04  510.97  1363.8
  520.28 1362.15  529.74 1362.69  535.98 1365.19  551.15 1371.27   572.4  1382.9
  592.61 1386.96  608.16  1387.7  613.78 1388.89  635.25 1390.77  676.52 1395.91
  709.15  1403.5  722.04 1407.25  766.93 1417.83  780.84 1420.34  824.49 1430.94
  850.36 1433.47  866.89 1437.06  880.84 1437.31  932.99 1443.36  955.65 1444.82
#Mann= 3 , 0 , 0
       0     .08       0  510.97    .055       0  535.98     .13       0
Bank Sta=510.97,535.98
Exp/Cntr=0.3,0.1

Type RM Length L Ch R = 1 ,240211.7,864.16,869.21,872.85
BEGIN DESCRIPTION:
52943.71
END DESCRIPTION:
XS GIS Cut Line= 3
  1097998.574929    688482.11715  1097645.543419   688123.828094
  1097292.600312   687748.989688
#Sta/Elev= 30
       0 1399.13  103.48 1383.52  129.54 1380.83  165.88 1375.18  185.45 1373.45
  248.39  1370.8  275.28 1370.94  290.15 1368.47  295.35 1366.46  440.23 1360.02
  468.09 1359.32  490.74 1357.05  502.99 1354.99  509.27    1356  515.72 1358.39
  524.99 1360.52  574.82 1362.48  630.06 1362.48   702.5 1364.41  762.88 1367.26
  784.54 1372.01  788.15 1372.04  797.53  1375.3   806.2 1377.48  822.79 1384.28
  834.03  1386.1  874.66 1395.88  972.76 1427.96  996.18 1434.15 1017.85 1438.94
#Mann= 3 , 0 , 0
       0     .08       0  490.74    .055       0  515.72     .08       0
Bank Sta=490.74,515.72
Exp/Cntr=0.3,0.1

Type RM Length L Ch R = 1 ,239342.5,1132.98,1130.79,1125.09
BEGIN DESCRIPTION:
52074.5
END DESCRIPTION:
XS GIS Cut Line= 3
  1098657.032032   688183.435578  1098033.520959   687319.634708
  1097500.460082   687342.562069
#Sta/Elev= 30
       0 1439.08  105.25 1414.49  202.12 1393.73  247.23 1385.21  411.26 1368.17
  420.13 1366.32  442.38 1366.09  502.14 1360.87  545.97 1358.99  598.65 1357.56
  767.01 1356.84  818.91 1355.91   843.6 1354.25  881.17 1354.96  925.86 1352.15
  938.59 1350.15  951.66 1352.95 1003.51  1354.8 1018.29 1364.65 1040.22 1381.46
 1055.63 1386.23 1096.08 1391.13 1115.71 1391.23  1206.9 1398.35 1252.75 1399.44
 1284.28 1402.54 1352.46 1403.25 1434.37 1406.45 1480.43 1406.58 1598.88 1413.36
#Mann= 3 , 0 , 0
       0     .08       0  925.86    .055       0  951.66     .09       0
Bank Sta=925.86,951.66
Exp/Cntr=0.3,0.1

Type RM Length L Ch R = 1 ,238211.7,909.83,912.66,908.19
BEGIN DESCRIPTION:
50943.71
END DESCRIPTION:
XS GIS Cut Line= 3
  1099546.288525   687504.613852  1098922.199451   686817.021389
  1098431.038128   686308.936266
#Sta/Elev= 30
       0 1440.19   47.33 1432.02  153.46 1426.18  195.21 1421.42  282.93 1404.51
  350.17 1386.01  415.98 1370.87  493.82 1357.79  538.97 1357.32  566.04  1353.4
  630.16 1350.59  765.04  1349.4  804.18 1347.16   895.5 1347.52  920.03 1344.25
  928.59 1341.85  938.58 1342.87  942.24 1346.82  944.57 1349.19  978.68 1352.63
  990.14 1357.06 1010.14 1369.75 1023.91 1372.54 1065.86 1375.63  1212.6 1394.71
 1286.91 1406.71 1308.43    1408 1329.88 1412.31 1437.94  1421.1 1635.26 1460.79
#Mann= 3 , 0 , 0
       0     .08       0  920.03    .055       0  942.24      .1       0
Bank Sta=920.03,942.24
Exp/Cntr=0.3,0.1

Type RM Length L Ch R = 1 ,237299.1,47.2,90.11,123.49
BEGIN DESCRIPTION:
50031.05
END DESCRIPTION:
XS GIS Cut Line= 4
  1099430.111187   686331.757009  1099393.692453   686157.467456
  1099305.247028   686063.819304  1099125.754748   685889.529706
#Sta/Elev= 30
       0 1346.24   48.26 1346.24  141.19 1344.11  172.08 1342.54  192.33 1342.76
  203.97 1342.18  217.04 1340.03  222.08 1338.74  236.08 1337.56     243 1338.31
  249.23 1342.17  258.15 1345.51  271.33 1348.21  289.26 1348.47   311.8 1351.59
  322.36  1351.8  333.05 1353.78  342.77 1357.95  347.54 1358.12  353.18 1359.63
  375.07 1360.53  385.46 1367.08  406.12 1368.74  426.92 1379.63   436.5 1380.96
  476.46  1393.1  486.92 1394.49   498.5 1399.78  510.85 1404.12  557.05 1418.44
#Mann= 3 , 0 , 0
       0     .09       0  217.04    .055       0  249.23     .12       0
Bank Sta=217.04,249.23
Exp/Cntr=0.5,0.3

Type RM Length L Ch R = 1 ,237209.0,115.53,96.02,84.96
BEGIN DESCRIPTION:
49940.94  Upstream xs of Bridge 37111-0362
END DESCRIPTION:
XS GIS Cut Line= 4
   1099437.91521   686352.567739  1099403.673035    686124.21345
  1099403.673035   685990.773799  1099296.188868   685581.566165
#Sta/Elev= 30
       0  1346.3 159.806  1346.7 168.999  1344.3 179.605  1338.5 183.848  1337.3
 193.747  1338.4  205.571338.559 222.739  1339.5 232.638  1346.2 279.378  1346.6
 300.733  1349.7 323.077  1352.1 332.764  1352.5 346.199  1352.2 352.281  1355.5
 365.998  1359.7 378.161  1361.8 384.737    1365 399.374  1368.4 406.021  1368.8
 419.385  1368.2 429.779  1370.2  440.74  1376.1 450.851  1379.7 460.892  1384.2
 470.933  1387.5 481.328  1389.5 502.611  1391.5 544.331  1393.4 556.776  1393.1
#Mann= 3 , 0 , 0
       0      .1       0 179.605    .055       0  205.57     .13       0
#XS Ineff= 2 , 0
       0 125.511  1349.9 266.933       0  1349.9
Permanent Ineff=
       F       F
Bank Sta=179.605,205.57
Skew Angle= 45
Exp/Cntr=0.5,0.3

Type RM Length L Ch R = 3 ,237151.4,,,
BEGIN DESCRIPTION:
49883.41  Bridge : 37111-0362
END DESCRIPTION:
Bridge Culvert--1,0,-1,-1, 0
Deck Dist Width WeirC Skew NumUp NumDn MinLoCord MaxHiCord MaxSubmerge Is_Ogee
47.5,20,2.6,45, 112, 113, , , 0.95, 0, 0,0,,
 -14.001 -13.647 -12.516  -4.879   -.707   4.667  10.677  13.647  17.748  21.001
  23.335  28.214  35.214  35.709  47.588  48.578  50.912  56.427  58.831  65.832
  70.781  76.297  82.378  86.196  93.762  94.399  94.752 101.187 106.773 107.975
 109.814 115.329 119.218 122.683 130.037 130.673 130.956 142.058 142.341 142.623
 159.099 159.099 233.345 233.345 249.326 254.346 259.862 266.791 268.913 270.185
 272.448 281.428 287.368 289.207 290.267 296.207 301.935 302.854 304.056 309.501
 313.955 316.996 324.279 325.906 326.542 336.795 339.411 348.179 351.856 357.937
 363.594 368.827  375.12 378.797 383.676 385.373 386.575 393.293 398.808 399.162
 402.627 410.688 414.506 421.931 426.739 432.891 432.961 432.961 440.174 443.427
 446.962 452.195 453.397 454.175 461.882 465.418 472.064 476.802  483.59  487.55
 494.197 498.227 506.147 508.763  515.41 518.946 522.905 529.482 530.047  530.33
  537.26  541.29
  1348.5  1348.5  1348.4  1348.2  1348.1    1348    1348    1348    1348  1347.9
  1347.9  1347.9  1348.1  1348.1  1348.2  1348.1  1348.1  1347.9  1347.9  1347.9
    1348    1348    1348  1348.2  1348.3  1348.3  1348.3  1348.4  1348.7  1348.6
  1348.7  1348.7  1348.7  1348.9  1348.9    1349    1349  1349.1  1349.1  1349.1
    1350    1350    1350    1350  1350.5  1350.7  1350.8  1350.8  1350.8  1350.7
  1350.9  1351.2  1351.4  1351.3  1351.4  1351.5  1351.9  1351.9    1352  1351.7
  1352.6  1352.6  1352.8  1352.7  1352.8  1353.2  1353.6  1354.4  1354.8  1355.2
  1356.2  1356.8  1357.5  1357.9  1358.5  1358.8  1358.8  1359.7  1360.9    1361
  1361.4  1362.3  1362.8  1363.9  1364.7  1365.5  1365.5  1365.5  1366.1  1366.8
  1367.3  1367.9  1367.9  1368.1    1369  1369.6  1370.3  1370.9  1371.6    1372
  1372.8  1373.3  1373.9  1374.1  1374.9  1375.2  1375.5    1376    1376  1376.1
    1377  1377.4
                                                                                
                                                                                
                                                                                
                                                                                
          1347.7  1347.7
                                                                                
                                                                                
                                                                                
                                                                                
                                                                                
                                                                                
                
       0   5.445   5.798    6.93  14.637  18.738  24.112  30.123  33.093  37.194
  40.447   42.78  47.659  54.659  55.154  67.034  68.024  70.357  75.873  78.277
  85.277  90.227  95.742 101.823 105.642 113.208 113.844 114.198 120.632 126.219
 127.421 129.259 134.775 138.664 142.128 149.482 150.119 150.402 161.503 161.786
 162.069 180.312 180.312 254.558 254.558 268.771 273.792 279.307 286.237 288.358
 289.631 291.894 300.874 306.814 308.652 309.713 315.652  321.38 322.299 323.501
 328.946 333.401 336.441 343.725 345.351 345.987  356.24 358.857 367.625 371.302
 377.383  383.04 388.272 394.566 398.243 403.122 404.819 406.021 412.738 418.254
 418.607 422.072 430.133 433.951 441.376 446.184 452.336 452.407 452.407 459.619
 462.872 466.408  471.64 472.842  473.62 481.328 484.863  491.51 496.248 503.036
 506.996 513.642 517.673 525.592 528.209 534.856 538.391 542.351 548.927 549.493
 549.776 556.705 560.736
  1348.5  1348.5  1348.5  1348.4  1348.2  1348.1    1348    1348    1348    1348
  1347.9  1347.9  1347.9  1348.1  1348.1  1348.2  1348.1  1348.1  1347.9  1347.9
  1347.9    1348    1348    1348  1348.2  1348.3  1348.3  1348.3  1348.4  1348.7
  1348.6  1348.7  1348.7  1348.7  1348.9  1348.9    1349    1349  1349.1  1349.1
  1349.1    1350    1350    1350    1350  1350.5  1350.7  1350.8  1350.8  1350.8
  1350.7  1350.9  1351.2  1351.4  1351.3  1351.4  1351.5  1351.9  1351.9    1352
  1351.7  1352.6  1352.6  1352.8  1352.7  1352.8  1353.2  1353.6  1354.4  1354.8
  1355.2  1356.2  1356.8  1357.5  1357.9  1358.5  1358.8  1358.8  1359.7  1360.9
    1361  1361.4  1362.3  1362.8  1363.9  1364.7  1365.5  1365.5  1365.5  1366.1
  1366.8  1367.3  1367.9  1367.9  1368.1    1369  1369.6  1370.3  1370.9  1371.6
    1372  1372.8  1373.3  1373.9  1374.1  1374.9  1375.2  1375.5    1376    1376
  1376.1    1377  1377.4
                                                                                
                                                                                
                                                                                
                                                                                
                  1347.7  1347.7
                                                                                
                                                                                
                                                                                
                                                                                
                                                                                
                                                                                
                        
Pier Skew= 45
Pier Skew, UpSta & Num, DnSta & Num=  ,183.848, 2 ,205.061, 2 , 0 , 0 , 0 ,,
       1       1
  1336.3  1348.2
       1       1
  1336.3  1348.2
Pier Skew, UpSta & Num, DnSta & Num=  ,208.596, 2 ,229.81, 2 , 0 , 0 , 0 ,,
       1       1
  1337.6  1348.2
       1       1
  1337.6  1348.2
BR Coef=-1 , 1 , 0 ,, 0 ,,,0.8,0,1.2,0,
WSPro=,,,, 1 ,,,, 0 ,,,, 0 ,,,,-1 ,-1 ,-1 , 0 , 0 , 0 , 0 , 0
BC Design=,, 0 ,, 0 ,,,,,,

Type RM Length L Ch R = 1 ,237112.9,518.02,491.1,462.75
BEGIN DESCRIPTION:
49844.93  Down stream xs of Bridge 37111-0362
END DESCRIPTION:
XS GIS Cut Line= 5
  1099554.975389   686323.953029  1099503.682272    686110.60231
  1099482.609174   686065.011335  1099481.669471   685949.426303
  1099440.772479   685556.542077
#Sta/Elev= 30
       0  1345.2  38.608  1344.7 181.019  1346.7 190.212  1344.3 200.818  1338.5
 205.061  1337.3  214.96  1338.4  229.81  1338.6 243.952  1339.5 253.851  1346.2
 300.025  1344.4 363.311  1346.7 371.938  1347.3 379.575  1348.5 398.172  1350.2
 410.617  1352.1  415.92    1352 422.213  1353.1 430.557  1353.7 444.558  1355.7
 448.942  1356.9 456.367  1355.9 475.883  1358.6 478.641  1358.7 499.712  1362.7
 510.248  1362.3  522.34  1363.7 528.421    1365 543.482  1367.1 551.755  1366.9
#Mann= 3 , 0 , 0
       0     .12       0 200.818    .054       0  229.81     .12       0
#XS Ineff= 2 , 0
       0  160.16  1347.9 274.711       0  1347.9
Permanent Ineff=
       F       F
Bank Sta=200.818,229.81
Skew Angle= 45
Exp/Cntr=0.5,0.3

Type RM Length L Ch R = 1 ,236621.8,575,577.12,580
BEGIN DESCRIPTION:
49353.83
END DESCRIPTION:
XS GIS Cut Line= 2
  1100246.931052   686084.629989  1099536.766045   685520.139825
#Sta/Elev= 30
       0 1383.01   28.82 1377.04   50.68 1373.52   91.67 1370.96  112.72 1363.76
   118.4  1362.9  127.45 1358.71  145.67 1356.19  173.32  1349.3  195.98 1345.73
   209.9 1341.91     215 1341.36   279.6 1340.42   374.8 1337.33  396.32 1340.27
  418.09 1338.49  427.03    1337  461.26 1339.99  482.53 1338.74  500.45 1335.68
  514.59 1333.71  521.65 1334.73  523.98 1335.84   528.7 1337.99  536.84 1339.93
  547.87 1339.35   684.4 1343.83  791.11 1346.04  893.93 1357.73  907.18 1359.99
#Mann= 3 , 0 , 0
       0      .1       0  500.45    .054       0  523.98      .1       0
Bank Sta=500.45,523.98
Exp/Cntr=0.3,0.1

Type RM Length L Ch R = 1 ,236044.7,826.44,833,816.06
BEGIN DESCRIPTION:
48776.71
END DESCRIPTION:
XS GIS Cut Line= 4
  1100439.071359   685743.424704  1100172.011118   685485.417337
  1100140.325994   685394.888423  1099607.382484   685054.067361
#Sta/Elev= 30
       0  1345.1   12.77 1345.82   33.84 1350.09   45.48 1350.96   68.11 1350.74
   95.94  1348.2  119.94 1343.19  236.95 1338.28  312.22 1337.37  355.33 1335.66
  378.43 1337.41     398  1336.3  410.58  1333.1  423.76 1331.03  430.44 1332.07
  440.86 1336.08  450.22  1336.8  486.09 1335.51   528.7 1337.29  701.96 1340.62
  763.81 1343.33  844.62 1357.21  884.11 1369.12  916.35 1377.43  966.85 1387.48
   977.8 1392.34 1018.37 1402.44  1027.4 1405.75 1076.15 1418.54 1099.85 1426.68
#Mann= 3 , 0 , 0
       0      .1       0  410.58    .054       0  430.44      .1       0
Bank Sta=410.58,430.44
Exp/Cntr=0.3,0.1

Type RM Length L Ch R = 1 ,235211.7,999.54,1000,1001.38
BEGIN DESCRIPTION:
47943.71
END DESCRIPTION:
XS GIS Cut Line= 3
  1100969.740577   685565.373763  1100647.099584   684961.755175
  1100272.995908   684380.362579
#Sta/Elev= 30
       0 1365.65   34.05 1367.14   50.79 1366.16   164.1 1353.01   223.7 1348.44
   266.6 1342.56  310.36 1343.81  468.43 1336.48  585.08 1335.08  622.43 1332.84
  639.29 1333.73  669.27 1328.82  684.44 1326.69  700.15 1328.52  726.18 1332.77
  776.09 1333.19  847.45 1338.41  871.21  1348.5  935.72 1363.98  950.98 1365.36
 1027.66 1387.99 1050.72 1390.85 1074.46 1397.57 1103.95 1402.71 1148.25 1406.52
 1214.62 1417.62 1240.03 1427.27 1264.68 1440.74 1351.19 1476.01 1375.79  1488.3
#Mann= 3 , 0 , 0
       0     .08       0  669.27    .054       0  700.15     .08       0
Bank Sta=669.27,700.15
Exp/Cntr=0.3,0.1

Type RM Length L Ch R = 1 ,234211.7,1190.86,1183.95,1172.4
BEGIN DESCRIPTION:
46943.71
END DESCRIPTION:
XS GIS Cut Line= 3
  1101827.454636   685053.127481  1101443.765397   684460.457919
  1101130.805168   683852.960664
#Sta/Elev= 30
       0 1391.68    11.6 1389.06  173.05 1372.16  398.26 1355.82  540.55 1344.23
  557.78 1339.18  584.11 1339.86  602.87 1335.51  618.63 1333.58  669.84 1330.18
  692.34 1322.56  706.03 1320.12  713.53 1321.15  721.04 1324.17  729.07 1325.67
   747.1 1323.66  763.39    1328  771.51 1328.36  983.13 1332.71 1040.58 1337.89
 1081.94 1350.24 1095.24 1358.34 1133.36 1367.34 1190.17 1387.46  1208.7 1395.39
 1235.57    1404 1291.17 1426.04 1352.85 1452.81 1377.07 1459.29  1389.4 1464.71
#Mann= 3 , 0 , 0
       0     .11       0  692.34    .054       0  721.04     .11       0
Bank Sta=692.34,721.04
Exp/Cntr=0.3,0.1

Type RM Length L Ch R = 1 ,233027.8,540.27,565.74,588.99
BEGIN DESCRIPTION:
45759.76
END DESCRIPTION:
XS GIS Cut Line= 3
  1102778.303437   684132.867728   1102262.84094    683685.22504
  1101757.695181   683226.326533
#Sta/Elev= 30
       0 1365.07   52.12 1359.23   75.92 1358.03  135.12 1352.41  222.53 1341.81
  238.56  1338.4   320.3  1332.9  356.22 1330.64  462.77 1326.57  700.81 1323.35
  722.45 1321.53  726.73 1320.16  757.96 1315.93   773.2 1313.95  780.81 1314.96
  788.45 1320.15  809.06 1321.88  902.85  1324.1  960.13 1327.09  978.77 1329.01
  996.17 1332.78 1075.43  1359.8 1094.13 1364.84 1128.35 1378.37  1186.7 1398.29
 1201.23 1401.35 1278.88 1425.71  1323.4 1437.36 1343.06 1440.66 1365.17 1442.19
#Mann= 3 , 0 , 0
       0     .08       0  757.96    .054       0  788.45     .08       0
Bank Sta=757.96,788.45
Exp/Cntr=0.3,0.1

Type RM Length L Ch R = 1 ,232462.0,95.43,109.05,123.41
BEGIN DESCRIPTION:
45194.02
END DESCRIPTION:
XS GIS Cut Line= 4
  1102705.795909   683604.583195  1102500.012921   683279.831925
  1102493.582179   683160.863643  1102239.568804   682990.449558
#Sta/Elev= 30
       0 1330.43  101.92 1324.86  190.63 1323.02   273.8 1322.28  315.51 1319.77
  413.64 1318.75  424.28 1316.73  430.03 1313.98  436.41 1310.07  439.64 1309.64
  442.12 1310.15  454.32 1316.76  456.77 1316.83  464.03 1319.25  470.29 1323.96
  486.08 1331.08   503.6 1339.63  509.66  1341.7  515.07 1344.22  551.45 1363.21
  570.45 1372.02  576.34 1375.59  612.74 1394.61   635.1 1404.07  672.66 1415.66
  692.08 1420.97  723.79 1428.56  741.55 1431.85  752.78 1433.01  809.48 1436.24
#Mann= 3 , 0 , 0
       0     .12       0  424.28    .054       0  454.32     .12       0
Bank Sta=424.28,454.32
Exp/Cntr=0.5,0.3

Type RM Length L Ch R = 1 ,232353.0,127.72,139.65,153.05
BEGIN DESCRIPTION:
45084.97
END DESCRIPTION:
XS GIS Cut Line= 6
  1102725.886969   683613.870806  1102658.208649   683424.371511
  1102588.993523   683234.551164  1102608.122757    683147.34446
  1102270.273312   682894.051156 1102236.1087508  682868.4372184
#Sta/Elev= 30
       0  1337.7 114.559  1332.4 149.912  1331.8 168.457  1330.2  204.68  1329.8
 347.637  1324.4 368.404  1323.4 379.416  1321.9 393.518  1323.5 418.342  1322.8
 427.905  1309.5 446.258    1308 460.747  1309.8 483.446    1315 503.634    1316
 518.509    1319 529.714  1318.3 560.334  1327.6 583.999  1329.5 635.386  1330.5
 647.846  1332.2 669.676  1331.1 694.018  1332.7 703.291  1331.3 741.638  1332.4
 806.838  1331.5 824.514  1333.5   839.1  1332.7 847.407    1334 924.874  1334.4
#Mann= 3 , 0 , 0
       0     .12       0 427.905    .054       0 460.747     .12       0
#XS Ineff= 2 , 0
           404.6 1316.89  521.48         1317.12
Permanent Ineff=
       F       F
Bank Sta=427.905,460.747
Skew Angle= 15
Exp/Cntr=0.5,0.3

Type RM Length L Ch R = 3 ,232289.2,,,
BEGIN DESCRIPTION:
45021.22  Bridge: 37111-0363
END DESCRIPTION:
Bridge Culvert--1,0,-1,-1, 0
Deck Dist Width WeirC Skew NumUp NumDn MinLoCord MaxHiCord MaxSubmerge Is_Ogee
60,20,2.6,15, 97, 97, , , 0.95, 0, 0,0,,
       0  15.068  22.023  37.864  39.989  55.831  58.632    65.2   77.95  90.604
  93.115  95.047  96.303 111.468  122.19  129.82 144.696 146.434 147.304 163.048
 174.929 181.497 188.162 194.441 201.299 207.094 215.112 224.771 232.692 235.783
 260.607 265.919 281.374 283.886 297.892 300.403 300.886 318.949 328.801 338.943
 344.739 349.569 359.904 362.512 374.007 384.825 386.467 388.592 425.973 425.973
 480.065 480.065 571.055 573.374 580.618 589.215 589.987 591.147 598.294  600.13
 612.397 623.312  625.92  630.46 637.608 645.238 650.068 654.415 657.892 662.625
 664.364 665.909 674.216 683.875 684.069 684.165 692.762 693.535 705.995 716.524
 719.132 723.961 731.399 737.967  742.99 748.496 752.456 757.865 760.763 762.598
 771.485  778.44  782.11 791.093 792.349  803.94 816.787
  1356.7  1356.7  1355.8  1354.2  1353.9  1354.9    1355    1355  1354.9  1354.7
  1354.7  1354.6  1354.6  1354.4  1354.5  1354.5  1353.9  1353.9  1353.9    1354
  1353.5  1353.2  1352.8  1352.4  1351.9  1351.7  1351.3  1350.4  1349.6  1349.1
  1346.3  1345.8  1342.9  1342.4  1338.6  1337.9  1337.7  1331.7  1329.6  1326.1
  1325.5  1325.3  1324.8  1324.5  1323.1  1321.4  1321.2  1321.1    1320    1320
    1320    1320  1314.9  1313.5    1314  1312.4  1312.3  1312.2  1311.6    1312
  1312.9  1312.5  1312.6  1312.8  1313.5  1314.4  1314.8  1314.5    1314  1314.3
  1314.3  1314.4  1314.8  1314.8  1314.8  1314.8  1315.1  1315.1  1316.2  1316.1
  1316.1  1316.3  1316.3  1316.4  1316.5  1316.5  1316.5  1316.5  1316.5  1316.5
  1316.5  1316.5  1316.5  1316.6  1316.6  1316.9  1316.9
                                                                                
                                                                                
                                                                                
                                                                                
                                                                          1317.9
  1317.9
                                                                                
                                                                                
                                                                                
                                                        
       0  75.052  82.104  97.945  99.973 115.911 118.712 125.281 138.031 150.684
 153.196 155.031 156.383 171.548 182.174 189.804  204.68 206.418 207.288 223.129
 234.913 241.481 248.243 254.521  261.38 267.078 275.096 284.755 292.772 295.767
 320.687 325.903 341.358  343.87 357.972 360.387  360.87 379.029 388.882 398.927
 404.723 409.553 419.888 422.496 434.087 444.905 446.451 448.576 486.054 486.054
 540.146 540.146 631.039 633.454 640.699 649.199 649.971 651.131 658.375  660.21
 672.478 683.296 686.001  690.54 697.592 705.319 710.052 714.399 717.876 722.609
 724.444 725.893   734.2 743.956 744.053 744.246 752.746 753.615 766.076 776.604
 779.212 784.042 791.383 798.048 802.974 808.576  812.44 817.946 820.747 822.582
 831.566  838.52 842.191 851.174 852.333 863.924 876.867
  1356.7  1356.7  1355.8  1354.2  1353.9  1354.9    1355    1355  1354.9  1354.7
  1354.7  1354.6  1354.6  1354.4  1354.5  1354.5  1353.9  1353.9  1353.9    1354
  1353.5  1353.2  1352.8  1352.4  1351.9  1351.7  1351.3  1350.4  1349.6  1349.1
  1346.3  1345.8  1342.9  1342.4  1338.6  1337.9  1337.7  1331.7  1329.6  1326.1
  1325.5  1325.3  1324.8  1324.5  1323.1  1321.4  1321.2  1321.1    1320    1320
    1320    1320  1314.9  1313.5    1314  1312.4  1312.3  1312.2  1311.6    1312
  1312.9  1312.5  1312.6  1312.8  1313.5  1314.4  1314.8  1314.5    1314  1314.3
  1314.3  1314.4  1314.8  1314.8  1314.8  1314.8  1315.1  1315.1  1316.2  1316.1
  1316.1  1316.3  1316.3  1316.4  1316.5  1316.5  1316.5  1316.5  1316.5  1316.5
  1316.5  1316.5  1316.5  1316.6  1316.6  1316.9  1316.9
                                                                                
                                                                                
                                                                                
                                                                                
                                                                          1317.9
  1317.9
                                                                                
                                                                                
                                                                                
                                                        
Pier Skew= 15
Pier Skew, UpSta & Num, DnSta & Num=  ,460.747, 2 ,520.827, 2 , 0 , 0 , 0 ,,
       3       3
    1308  1317.9
       3       3
    1308  1317.9
BR Coef=-1 , 1 , 0 ,, 0 ,,,0.8,0,2,0,
WSPro=,,,, 1 ,,,, 0 ,,,, 0 ,,,,-1 ,-1 ,-1 , 0 , 0 , 0 , 0 , 0
BC Design=,, 0 ,, 0 ,,,,,,

Type RM Length L Ch R = 1 ,232213.3,434.08,386.36,335.83
BEGIN DESCRIPTION:
44945.32
END DESCRIPTION:
XS GIS Cut Line= 4
   1102863.34851   683492.045655  1102686.371432    683194.35434
   1102717.13991   683058.093849  1102817.345927  682756.9463017
#Sta/Elev= 30
       0  1358.3  11.591  1357.2  50.615  1350.3  70.609    1348  87.416  1344.9
 105.093  1340.5 136.485  1334.1 193.572  1323.5 224.288  1320.2  290.55  1316.5
 338.847    1315 376.518  1311.6 487.503  1310.8 487.986  1309.5 506.338    1308
 520.827  1309.8 536.282  1312.8 545.072  1311.1 569.027    1311 648.426  1316.5
 663.398  1316.9 684.165  1319.8  686.58  1320.8 690.057  1323.5 706.768  1333.8
 731.206  1334.6 745.405  1337.3 751.683  1340.3 766.849  1349.3 776.025  1352.7
#Mann= 3 , 0 , 0
       0     .12       0 487.986    .053       0 520.827     .12       0
#XS Ineff= 2 , 0
          472.33 1315.87  552.25         1315.97
Permanent Ineff=
       F       F
Bank Sta=487.986,520.827
Skew Angle= 15
Exp/Cntr=0.5,0.3

Type RM Length L Ch R = 1 ,231827.0,604.47,615.25,620.62
BEGIN DESCRIPTION:
44558.96
END DESCRIPTION:
XS GIS Cut Line= 2
  1103324.593186   683180.190075  1102746.114411   682622.670717
#Sta/Elev= 30
       0 1358.26   12.01 1357.16   52.39 1350.26   73.07 1348.02  141.29 1334.13
  200.44 1323.45  232.17 1320.24  305.44  1316.3  350.79 1314.98  389.83  1311.6
  504.65 1310.77  516.45 1308.91  531.16 1306.98  538.87 1308.02  543.89 1309.52
  546.59 1310.32  564.28 1311.09   589.1 1311.02  669.83 1316.43  686.81 1316.94
  708.26 1319.81  710.81 1320.75  714.38 1323.52  731.65 1333.77  743.69 1334.62
  757.03 1334.56  771.68 1337.26  778.22 1340.28  793.87 1349.32  803.41 1352.69
#Mann= 3 , 0 , 0
       0     .08       0  516.45    .053       0  543.89     .08       0
Bank Sta=516.45,543.89
Exp/Cntr=0.3,0.1

Type RM Length L Ch R = 1 ,231211.7,978.98,1000,1006.45
BEGIN DESCRIPTION:
43943.71
END DESCRIPTION:
XS GIS Cut Line= 3
  1103670.840605   683017.846204  1103340.092128   682417.061605
  1102981.714446   681817.225639
#Sta/Elev= 30
       0 1324.08   29.95 1322.69   35.32 1323.73    54.8 1323.31   76.51 1325.81
  110.77 1327.24   137.4 1332.03  176.64 1332.71  222.81 1329.41  312.48 1318.37
  354.04 1314.92  425.92 1311.58  568.77 1309.86  644.28 1307.31  663.74 1308.82
  670.88 1307.26  678.22 1304.21  685.81 1303.25  703.28 1305.39  711.77 1308.15
  753.22 1307.78  853.12  1310.1  984.66 1319.48 1101.57 1332.04 1131.18 1338.86
 1164.23 1338.65 1183.41 1342.41 1243.88 1349.54 1283.88 1352.28 1384.55  1364.8
#Mann= 3 , 0 , 0
       0     .08       0  670.88    .053       0  703.28     .08       0
#XS Ineff= 2 , 0
          549.37 1310.87
Permanent Ineff=
       F       F
Bank Sta=670.88,703.28
Exp/Cntr=0.3,0.1

Type RM Length L Ch R = 1 ,230211.7,490.67,482.48,473.14
BEGIN DESCRIPTION:
42943.71
END DESCRIPTION:
XS GIS Cut Line= 3
  1104271.956918   682826.500644   1104190.24583   682154.250218
  1104096.329401   681470.587332
#Sta/Elev= 30
       0 1325.18   24.66  1317.1   36.65 1314.82   63.53 1313.46  148.23 1311.14
  161.64 1309.52   178.5 1308.59   224.4 1307.57  299.08 1307.53  383.78 1306.24
  467.23 1306.51  543.31  1304.9   591.8 1302.66  634.73 1303.72  644.33 1301.34
  661.71 1299.59   677.2 1297.65  685.13 1298.71  693.13 1301.77  708.31 1303.89
  715.94  1304.2   759.3 1303.96  807.21 1308.01  874.26 1316.59   927.1 1326.55
  984.88 1329.73 1022.22 1330.81 1070.69  1330.8 1208.64 1329.07 1367.28 1332.42
#Mann= 3 , 0 , 0
       0     .09       0  661.71    .053       0  693.13     .09       0
Bank Sta=661.71,693.13
Exp/Cntr=0.3,0.1

Type RM Length L Ch R = 1 ,229729.2,302.02,312.55,322.98
BEGIN DESCRIPTION:
42461.23
END DESCRIPTION:
XS GIS Cut Line= 4
   1104721.82623   682488.853506  1104657.519033    682090.14897
  1104606.949628   681972.048824  1104570.270748   681489.983199
#Sta/Elev= 30
       0 1304.06  117.97 1304.18   231.7  1303.7  322.28 1302.26  373.12 1300.23
  427.24 1302.26  445.08 1298.91  452.54 1295.42  460.46 1294.37  476.11 1296.29
  491.34 1299.58  502.57 1300.22  510.66 1299.71  521.73 1300.36  529.74    1301
  542.23  1302.8  572.81 1304.55  632.98 1305.93  649.08  1306.7  696.33 1307.07
  734.82 1306.64  780.37  1308.6  826.22 1311.28  866.03 1314.68  910.68 1319.81
   962.5 1327.24  982.26 1330.45   993.4 1332.78 1002.35 1333.59 1015.79 1333.15
#Mann= 3 , 0 , 0
       0     .09       0  445.08    .053       0  476.11     .09       0
#XS Ineff= 2 , 0
           312.5 1304.57
Permanent Ineff=
       F       F
Bank Sta=445.08,476.11
Exp/Cntr=0.5,0.3

Type RM Length L Ch R = 1 ,229416.7,69.91,69.62,68.53
BEGIN DESCRIPTION:
42148.68
END DESCRIPTION:
XS GIS Cut Line= 3
  1104957.425243   682440.135032  1104920.753737   681911.016881
  1104889.323163    681518.13461
#Sta/Elev= 30
       0 1302.55 213.497 1302.23 265.306 1301.71 321.932 1299.73 332.835  1299.5
 339.524 1299.76 348.851 1297.41  354.09 1294.11  366.54 1294.11 370.057  1297.6
 375.042 1299.81 382.121 1300.69 387.289 1300.77 396.333 1299.51 458.474 1300.24
 534.643 1305.04 547.951 1306.18 557.299 1306.64 558.529 1306.98 569.773 1307.38
 584.063 1310.31  589.14 1310.41 596.402 1314.24 601.055 1315.66 604.562 1317.76
 618.238 1319.57 630.138 1319.89 637.641 1323.72 645.327 1328.32 653.734 1332.62
#Mann= 3 , 0 , 0
       0     .09       0 348.851    .053       0 370.057     .09       0
#XS Ineff= 2 , 0
       0 346.136 1298.79  372.27       0 1298.79
Permanent Ineff=
       F       F
Bank Sta=348.851,370.057
Skew Angle= 45
Exp/Cntr=0.5,0.3

Type RM Length L Ch R = 2 ,229381.1,,,
BEGIN DESCRIPTION:
42113.1  Culvert: 37111-0365
END DESCRIPTION:
Bridge Culvert--1,0,-1,-1, 0
Deck Dist Width WeirC Skew NumUp NumDn MinLoCord MaxHiCord MaxSubmerge Is_Ogee
25,18,2.6,45, 125, 125, 1298.79, , 0.95, 0, 0,0,,
       0   2.376   5.339    6.47   8.174  13.039  20.237  23.511  28.489  31.198
  37.717  41.295  45.884   47.85  54.207  58.004  71.496  75.074  92.631  94.936
 109.213 111.398 115.704 118.766 125.709 128.276 133.834 137.391 150.833 165.774
 167.386 174.606 177.625 182.971 185.113 190.968 194.327 200.033 201.349 203.866
 216.254 217.407 220.681 235.318 235.375 246.024 246.087 265.915 268.863 271.967
 297.657 300.322 304.622 307.528 314.627 316.218 320.864 323.466 338.188 346.235
 347.069 391.971 400.251 401.516 402.952 410.532 424.964 427.595 432.269 441.213
 443.603 456.084 457.053 457.668   462.9 470.558 471.619 477.007 478.471  484.92
 487.197 492.295 493.744 499.422 502.626 506.501 508.155 511.846  516.93 521.569
 524.263  532.14 532.925 533.031  533.47 538.674 539.989 546.707 548.955 553.353
 555.411 560.212 565.205 568.655 572.905 579.983 582.119 583.893 589.197 593.814
 598.439 601.684 605.743 608.699 615.423 616.456 623.117 628.165 632.627  636.46
   639.5 641.537 648.679 651.005  653.89
 1303.36  1303.3 1303.05 1303.09 1303.13  1303.1 1303.07 1302.99 1302.82  1302.8
 1302.84 1302.84 1302.79 1302.79  1302.7  1302.7 1302.63 1302.69 1302.67 1302.68
 1302.73 1302.77 1302.75 1302.71 1302.86  1302.8 1302.48 1302.49 1302.46 1302.43
 1302.48 1302.52 1302.48 1302.45 1302.44 1302.37 1302.39 1302.66 1302.66 1302.67
 1302.73 1302.73 1302.77 1302.94 1302.94 1302.93 1302.94 1302.58 1302.52 1302.47
 1301.52  1301.4  1301.3 1301.21  1301.1 1301.02 1300.68 1300.57 1299.31 1298.91
 1298.88 1298.79 1298.82 1298.82 1298.93 1298.84 1298.92 1299.07 1299.17 1299.52
 1299.74 1300.44 1300.43  1300.5  1300.6 1301.37 1301.45 1301.57 1301.71 1301.91
 1302.11 1302.62 1302.73 1302.82 1303.18 1303.84 1303.99 1304.39 1304.61 1305.25
 1305.42 1306.25  1306.3 1306.31 1306.33 1306.23 1306.38 1306.93  1307.1 1307.63
 1307.87 1308.31 1308.88 1309.49 1309.91 1311.28 1311.67 1311.88 1312.59 1313.52
 1316.38 1317.34 1317.89 1318.54 1318.59 1318.62 1319.47 1321.95 1324.34 1326.51
 1327.73 1328.64 1331.31 1333.22 1334.38
                                                                                
                                                                                
                                                                                
                                                                                
                                                                                
                                                                                
                                                                                
                                                                                
                                                                                
                                                                                
                                                                                
                                                                                
                                        
       0   2.376   5.339    6.47   8.174  13.039  20.237  23.511  28.489  31.198
  37.717  41.295  45.884   47.85  54.207  58.004  71.496  75.074  92.631  94.936
 109.213 111.398 115.704 118.766 125.709 128.276 133.834 137.391 150.833 165.774
 167.386 174.606 177.625 182.971 185.113 190.968 194.327 200.033 201.349 203.866
 216.254 217.407 220.681 235.318 235.375 246.024 246.087 265.915 268.863 271.967
 297.657 300.322 304.622 307.528 314.627 316.218 320.864 323.466 338.188 346.235
 347.069 391.971 400.251 401.516 402.952 410.532 424.964 427.595 432.269 441.213
 443.603 456.084 457.053 457.668   462.9 470.558 471.619 477.007 478.471  484.92
 487.197 492.295 493.744 499.422 502.626 506.501 508.155 511.846  516.93 521.569
 524.263  532.14 532.925 533.031  533.47 538.674 539.989 546.707 548.955 553.353
 555.411 560.212 565.205 568.655 572.905 579.983 582.119 583.893 589.197 593.814
 598.439 601.684 605.743 608.699 615.423 616.456 623.117 628.165 632.627  636.46
   639.5 641.537 648.679 651.005  653.89
 1303.36  1303.3 1303.05 1303.09 1303.13  1303.1 1303.07 1302.99 1302.82  1302.8
 1302.84 1302.84 1302.79 1302.79  1302.7  1302.7 1302.63 1302.69 1302.67 1302.68
 1302.73 1302.77 1302.75 1302.71 1302.86  1302.8 1302.48 1302.49 1302.46 1302.43
 1302.48 1302.52 1302.48 1302.45 1302.44 1302.37 1302.39 1302.66 1302.66 1302.67
 1302.73 1302.73 1302.77 1302.94 1302.94 1302.93 1302.94 1302.58 1302.52 1302.47
 1301.52  1301.4  1301.3 1301.21  1301.1 1301.02 1300.68 1300.57 1299.31 1298.91
 1298.88 1298.79 1298.82 1298.82 1298.93 1298.84 1298.92 1299.07 1299.17 1299.52
 1299.74 1300.44 1300.43  1300.5  1300.6 1301.37 1301.45 1301.57 1301.71 1301.91
 1302.11 1302.62 1302.73 1302.82 1303.18 1303.84 1303.99 1304.39 1304.61 1305.25
 1305.42 1306.25  1306.3 1306.31 1306.33 1306.23 1306.38 1306.93  1307.1 1307.63
 1307.87 1308.31 1308.88 1309.49 1309.91 1311.28 1311.67 1311.88 1312.59 1313.52
 1316.38 1317.34 1317.89 1318.54 1318.59 1318.62 1319.47 1321.95 1324.34 1326.51
 1327.73 1328.64 1331.31 1333.22 1334.38
                                                                                
                                                                                
                                                                                
                                                                                
                                                                                
                                                                                
                                                                                
                                                                                
                                                                                
                                                                                
                                                                                
                                                                                
                                        
Pier Skew= 45
BR Coef=-1 , 1 , 0 ,, 0 ,,,0.8,0,1.2,0,
WSPro=,,,, 1 ,,,, 0 ,,,, 0 ,,,,-1 ,-1 ,-1 , 0 , 0 , 0 , 0 , 0
Multiple Barrel Culv=1,3.5,,34,0.024,0.9,1,2,3,1294.11,1293.22, 3,Culvert #1  , 0 ,18
  356.17  375.03  360.17  379.03  364.17  383.03
Culvert Bottom n=0.024
BC Design=,, 0 ,, 0 ,,,,,,

Type RM Length L Ch R = 1 ,229347.1,462.32,472.32,482.4
BEGIN DESCRIPTION:
42079.06
END DESCRIPTION:
XS GIS Cut Line= 3
   1105022.20578   682437.369366  1104985.519525   681908.039045
   1104954.07198   681514.944783
#Sta/Elev= 30
       0 1301.23 231.535 1301.66 272.865 1301.21 342.678 1298.67  355.42 1299.11
 361.317 1299.94 366.861 1298.94 367.879 1298.17  373.23 1293.22  385.21 1293.22
 390.387 1296.23 399.777  1297.6 409.012 1297.26 430.621 1297.85 439.184 1298.57
 446.517 1297.76 474.264 1299.34 489.558 1300.47 518.776 1303.59 558.353 1306.46
  579.99  1309.2 590.724 1311.68 596.466 1314.74 601.154 1315.92 603.608 1317.45
 620.847 1318.54 628.236 1323.45 637.315 1325.35 647.038 1331.35 654.038 1334.96
#Mann= 3 , 0 , 0
       0     .09       0 367.879    .052       0 390.387     .09       0
#XS Ineff= 2 , 0
       0 362.385 1298.79 399.119       0 1298.79
Permanent Ineff=
       F       F
Bank Sta=367.879,390.387
Skew Angle= 45
Exp/Cntr=0.5,0.3

Type RM Length L Ch R = 1 ,228874.8,428.99,420.16,410.68
BEGIN DESCRIPTION:
41606.74
END DESCRIPTION:
XS GIS Cut Line= 4
  1105481.408148   682832.931342  1105429.205314   682051.564652
   1105458.14352   681942.242438   1105458.14352   681527.461047
#Sta/Elev= 30
       0 1353.59   25.95 1352.24    49.3 1352.39   62.95 1351.01   88.33    1345
  116.19 1347.05  253.98 1333.55  285.01 1333.22  361.38 1328.52  431.46 1320.18
  475.62 1312.54   535.2 1305.41  567.57 1302.81  623.88 1299.82  772.54 1296.04
  823.52 1291.81   839.6 1289.62  855.73 1291.86  911.79 1296.96  947.58 1297.09
   982.4 1298.73 1109.97 1307.41    1148  1311.2 1177.18 1311.44  1188.2 1313.76
 1199.69 1318.27 1240.42 1325.64 1271.69 1333.92  1284.5 1335.93 1310.98 1342.64
#Mann= 3 , 0 , 0
       0     .09       0  823.52    .052       0  855.73     .09       0
Bank Sta=823.52,855.73
Exp/Cntr=0.3,0.1

Type RM Length L Ch R = 1 ,228454.6,930.76,900.86,864.48
BEGIN DESCRIPTION:
41186.59
END DESCRIPTION:
XS GIS Cut Line= 4
  1106293.293164   682759.181671  1105862.332787   682227.771904
  1105849.371571    681916.70272  1105846.131278   681582.951441
#Sta/Elev= 30
       0 1349.29   50.73 1343.51   63.05 1339.58   79.81 1336.52  122.03 1335.09
  166.14 1329.95  235.02 1324.24  339.12 1320.01  402.56 1315.79   425.8    1313
  474.29 1312.71  522.08 1306.78   582.1 1303.45  747.09 1299.77  827.89 1296.23
  901.41 1295.24  913.42 1293.15  930.42 1286.99  935.88 1287.64  946.34 1292.94
  962.28 1294.52  1060.2 1295.16  1123.6 1299.26 1142.46 1301.47 1154.17 1305.23
 1178.22 1306.34 1206.07 1320.64 1214.75 1321.06 1283.76 1345.65  1329.3 1366.47
#Mann= 3 , 0 , 0
       0     .09       0  913.42    .052       0  946.34     .09       0
Bank Sta=913.42,946.34
Exp/Cntr=0.3,0.1

Type RM Length L Ch R = 1 ,227553.7,149.81,135.31,120.11
BEGIN DESCRIPTION:
40285.73
END DESCRIPTION:
XS GIS Cut Line= 4
  1106863.586579   682312.019786  1106649.726582   682000.950646
  1106562.238363    681958.82666  1106520.114422   681838.935468
#Sta/Elev= 30
       0 1360.05   43.61 1349.82   62.97  1346.1   92.47 1339.67  128.67 1333.49
  153.45 1328.27  160.69 1327.24  223.79 1315.43     234 1311.02  259.31 1302.64
  262.17 1302.81  272.23 1300.06  339.62 1293.33  361.06    1292  390.85  1291.4
   398.9 1290.67  409.12 1288.96  416.29 1287.05  422.14 1284.42  425.62 1283.87
  427.92  1284.3  442.67 1290.02  451.88 1290.52  465.02 1292.16  474.56 1291.12
   495.9 1292.01  542.71 1291.31  579.53 1293.63  591.82 1297.27  601.67 1297.13
#Mann= 3 , 0 , 0
       0     .09       0  409.12    .052       0  442.67     .09       0
Bank Sta=409.12,442.67
Exp/Cntr=0.5,0.3

Type RM Length L Ch R = 1 ,227418.4,100.12,80.64,79.35
BEGIN DESCRIPTION:
40150.41
END DESCRIPTION:
XS GIS Cut Line= 5
  1107156.087473   681864.988551   1106716.03464   681863.929925
  1106628.860721   681865.911151  1106553.475045   681869.194846
  1106545.864177   681841.469596
#Sta/Elev= 30
       0  1352.6   8.195 1351.93  18.314 1349.72  35.886 1343.16  49.625 1335.04
  69.862 1327.11  86.479 1319.16   94.88 1316.36  96.626 1314.75  98.168 1314.67
  100.36 1313.78 117.648 1304.57 123.631 1302.78 133.594  1297.9 140.453 1296.89
 147.856 1295.09 177.335 1292.27 277.384 1290.06 306.665 1290.45 319.082 1289.28
  320.49 1282.91  367.49 1282.91 371.125 1289.79 375.438 1289.98 383.224 1291.04
 410.801  1291.8  426.18  1292.6 430.282 1293.27 438.929 1295.88  446.51 1296.66
#Mann= 3 , 0 , 0
       0     .09       0 319.082    .051       0 371.125     .09       0
#XS Ineff= 2 , 0
       0  317.18 1293.63  373.13       0 1293.63
Permanent Ineff=
       F       F
Bank Sta=319.082,371.125
Skew Angle= 45
Exp/Cntr=0.5,0.3

Type RM Length L Ch R = 2 ,227375.4,,,
BEGIN DESCRIPTION:
40107.4  Culvert: 37111-0366
END DESCRIPTION:
Bridge Culvert--1,0,-1,-1, 0
Deck Dist Width WeirC Skew NumUp NumDn MinLoCord MaxHiCord MaxSubmerge Is_Ogee
17,47,2.6,45, 62, 61, , , 0.95, 0, 0,0,,
       0   5.713   6.442  11.278  16.313  19.926  34.945  40.192  44.088  49.936
  53.493  61.136  69.183  78.616  83.778  87.646  97.439 101.533 107.077  110.21
 114.049  118.37 125.695 144.914 147.128 154.934 163.943 170.144 177.081 177.901
 191.089 208.589  208.66  208.71 219.069 224.216 229.096 239.603 253.689 257.281
 267.965 268.241 268.559 283.253 285.402 291.703 299.834 310.342 315.794 375.467
 380.869 384.136 396.786 397.868   401.7 409.082  411.19 418.487 424.971 427.694
 433.379     450
 1326.32 1327.25 1327.07 1326.62 1325.77 1323.96  1316.1  1311.9 1310.13 1303.87
 1300.77 1298.72 1297.78 1294.82 1294.69 1294.58 1294.56 1294.64 1294.53 1294.43
 1294.33 1294.22  1294.1 1293.74 1293.61  1293.6 1293.65 1293.63 1293.67 1293.69
 1293.63  1293.8  1293.8  1293.8 1293.83 1293.85  1293.8 1293.97 1294.32 1294.31
 1294.31 1294.32 1294.32 1294.53 1294.55 1294.68 1294.77 1295.08 1295.08 1295.46
  1295.7 1295.81 1295.85  1295.9 1295.99 1296.18 1296.19 1296.04 1296.07 1296.18
 1296.31 1296.31
                                                                                
                                                                                
                                                                                
                                                                                
                                                                                
                                                                                
                
       0   5.713   6.442  11.278  16.313  19.926  34.945  40.192  44.088  49.936
  53.493  61.136  69.183  78.616  83.778  87.646  97.439 101.533 107.077  110.21
 114.049  118.37 125.695 144.914 147.128 154.934 163.943 170.144 177.081 177.901
 191.089 208.589  208.66  208.71 219.069 224.216 229.096 239.603 253.689 257.281
 267.965 268.241 268.559 283.253 285.402 291.703 299.834 310.342 315.794 375.467
 380.869 384.136 396.786 397.868   401.7 409.082  411.19 418.487 424.971 427.694
 433.379
 1326.32 1327.25 1327.07 1326.62 1325.77 1323.96  1316.1  1311.9 1310.13 1303.87
 1300.77 1298.72 1297.78 1294.82 1294.69 1294.58 1294.56 1294.64 1294.53 1294.43
 1294.33 1294.22  1294.1 1293.74 1293.61  1293.6 1293.65 1293.63 1293.67 1293.69
 1293.63  1293.8  1293.8  1293.8 1293.83 1293.85  1293.8 1293.97 1294.32 1294.31
 1294.31 1294.32 1294.32 1294.53 1294.55 1294.68 1294.77 1295.08 1295.08 1295.46
  1295.7 1295.81 1295.85  1295.9 1295.99 1296.18 1296.19 1296.04 1296.07 1296.18
 1296.31
                                                                                
                                                                                
                                                                                
                                                                                
                                                                                
                                                                                
        
Pier Skew= 45
BR Coef=-1 , 1 , 0 ,, 0 ,,,0.8,0,1.2,0,
WSPro=,,,, 1 ,,,, 0 ,,,, 0 ,,,,-1 ,-1 ,-1 , 0 , 0 , 0 , 0 , 0
Multiple Barrel Culv=2,10,15,50,0.013,0.2,1,8,1,1282.91,1282, 3,Culvert #1  , 0 ,15
  327.99  334.26  343.99  350.26  359.99  366.26
Culvert Bottom n=0.013
BC Design=,, 0 ,, 0 ,,,,,,

Type RM Length L Ch R = 1 ,227337.8,374.39,420.18,446.12
BEGIN DESCRIPTION:
40069.77
END DESCRIPTION:
XS GIS Cut Line= 5
  1107185.317411   681728.918195  1106997.368651   681741.093949
  1106763.286365   681783.969234  1106643.146797   681791.430748
  1106578.482163   681788.193565
#Sta/Elev= 30
       0  1308.7   5.728 1306.95  11.625 1307.28  20.301 1305.27  26.757 1299.87
   30.49 1296.27  33.255 1294.62   48.09 1294.72  75.378 1293.47 103.047 1291.13
 117.267 1290.39 143.295 1290.43 182.483 1289.32 221.614 1289.95 237.814 1289.99
 245.387 1289.62 290.614 1290.02 302.677 1290.24 308.581 1291.17 314.648 1291.54
 320.305 1291.01  326.76    1282  373.76    1282  374.13 1291.47 393.173 1296.17
 403.454 1300.85 413.438 1305.92 421.924 1309.64 428.089 1312.97 432.353 1314.21
#Mann= 3 , 0 , 0
       0     .08       0 320.305    .051       0  374.13     .12       0
#XS Ineff= 2 , 0
       0  314.69 1293.63  379.62       0 1293.63
Permanent Ineff=
       F       F
Bank Sta=320.305,374.13
Skew Angle= 45
Exp/Cntr=0.5,0.3

Type RM Length L Ch R = 1 ,226917.6,1240.46,1240.61,1238.44
BEGIN DESCRIPTION:
39649.59
END DESCRIPTION:
XS GIS Cut Line= 3
  1107505.105622   682039.038969  1107021.018346   681536.470918
  1105973.313174   680617.644775
#Sta/Elev= 30
       0 1368.79  127.67 1379.58  186.11  1374.9  262.51  1359.1  339.24 1333.51
  361.27 1331.04  393.85 1318.04  424.06 1312.82  466.41 1295.44  547.31 1289.67
  650.01 1288.75  671.51 1281.67  691.62 1291.11  780.53 1315.13  800.05 1325.27
     879 1344.92 1093.78 1372.88 1205.25 1374.46 1359.21 1389.07 1445.34 1387.67
 1538.06 1393.92 1580.56 1388.36 1634.39 1372.65 1658.58 1369.89 1689.54 1376.29
 1744.27 1374.93 1814.21 1393.38 1972.23 1403.13 2036.21  1394.8 2091.32 1382.92
#Mann= 3 , 0 , 0
       0     .08       0  650.01    .051       0  691.62     .13       0
Bank Sta=650.01,691.62
Exp/Cntr=0.3,0.1

Type RM Length L Ch R = 1 ,225677.0,718.37,712.8,704.89
BEGIN DESCRIPTION:
38408.98
END DESCRIPTION:
XS GIS Cut Line= 3
   1108446.80244   681177.914784  1107916.268227   680719.428488
  1106641.625805   679518.979311
#Sta/Elev= 30
       0 1373.31  209.03 1350.03  255.94 1341.18  380.22 1337.21  494.72 1344.12
  614.57 1334.91  682.08 1323.19  723.37 1310.36  780.38  1287.1  792.37 1284.99
  812.41 1279.58  832.27 1287.41  840.75 1289.04  892.09 1311.57  915.41 1319.21
  972.38 1332.89 1048.59 1343.19 1106.64 1346.99 1273.76 1335.75 1411.47 1331.86
 1488.41 1324.65  1509.1 1319.67 1530.07 1317.95 1652.95 1319.45 1702.69 1326.93
  2023.8 1388.81 2102.11 1395.25 2159.83 1404.52 2367.23 1428.35 2452.14 1431.44
#Mann= 3 , 0 , 0
       0     .14       0  792.37    .051       0  832.27     .13       0
Bank Sta=792.37,832.27
Exp/Cntr=0.3,0.1
