HEC-RAS study 2ndBroadRv.prj: 2ndBroadRv

--- 2ndBroadRv.g01 (geometry) --- (continued)

Type RM Length L Ch R = 1 ,207406.6,334.74,320.5,307.4
BEGIN DESCRIPTION:
20138.55  Down stream xs of Bridge 37111-0409
END DESCRIPTION:
XS GIS Cut Line= 4
  1117656.968633   672853.026286  1117664.959993   672792.027706
   1117682.53887   672660.186301  1117790.624051   672500.803872
#Sta/Elev= 30
       0  1125.3    8.21    1122  14.972  1120.2  20.381    1120  29.944  1117.4
  41.535  1112.8  45.495  1112.2  59.404  1106.1   78.24  1105.8  95.627  1099.3
 106.252  1090.8 116.877  1090.3 141.025    1090 159.378  1088.9  166.13 1086.71
 173.867  1084.2 188.356  1077.9 212.504  1078.3  234.72  1084.7 264.181  1095.2
 276.545  1096.1 291.323  1099.3 295.284  1099.3 304.943  1098.6 314.119  1098.9
 317.403  1098.6 333.824  1099.7 355.171  1100.4 368.597  1100.3  373.91  1099.9
#Mann= 3 , 0 , 0
       0     .13       0  166.13    .046       0  234.72     .13       0
#XS Ineff= 2 , 0
       0  57.898 1106.86 276.361       0  1108.4
Permanent Ineff=
       F       F
Bank Sta=166.13,234.72
Skew Angle= 15
Exp/Cntr=0.5,0.3

Type RM Length L Ch R = 1 ,207086.1,792.4,778.58,762.39
BEGIN DESCRIPTION:
19818.05
END DESCRIPTION:
XS GIS Cut Line= 4
   1118287.86441   672989.616404  1117987.191884   672660.497625
  1117959.165527    672528.89571  1117790.624051   672336.461716
#Sta/Elev= 30
       0  1179.4   39.46 1185.99   69.65 1187.34   97.96 1183.98  122.68 1178.21
  214.89 1148.85  248.21 1134.38  261.62 1123.68  270.45 1122.61   281.9 1124.28
  292.66 1121.62   329.2 1092.29  337.68 1089.79  443.97 1088.31  464.68 1090.47
  481.13 1086.42  505.61 1076.47  512.23 1077.12   530.7 1083.78  545.55 1088.18
  602.75 1088.15   649.8 1092.95  679.54 1091.47   736.3 1099.33  786.34 1103.31
  791.85 1104.68   798.8 1110.86  818.13 1110.12  827.65 1112.88  836.14  1112.2
#Mann= 3 , 0 , 0
       0     .13       0  481.13    .046       0   530.7     .13       0
Bank Sta=481.13,530.7
Exp/Cntr=0.3,0.1

Type RM Length L Ch R = 1 ,206307.5,68.47,55.23,41.95
BEGIN DESCRIPTION:
19039.47
END DESCRIPTION:
XS GIS Cut Line= 4
  1118582.837504   672370.172934  1118342.645129   672092.055405
  1118290.606487   672032.455961  1118005.533034   671995.135686
#Sta/Elev= 30
       0 1138.64   28.39 1131.36   59.86  1125.9   101.5 1113.75  112.81 1108.87
  142.26 1101.24  156.89 1098.14  182.51 1094.63  195.41  1091.6   235.3  1087.1
  259.23 1086.43  284.17 1083.15  361.26 1083.33  385.45 1076.39  395.84    1073
  407.94 1071.38  412.26  1071.7  420.48 1075.45   433.7 1084.84  454.29 1089.11
  473.27 1089.86  480.82 1091.43  524.32 1094.46  561.59 1095.55  577.57 1094.64
  594.99 1096.76  654.58 1094.41  662.36  1092.7  688.25 1090.81  734.11  1105.4
#Mann= 3 , 0 , 0
       0     .13       0  385.45    .046       0  420.48     .13       0
Bank Sta=385.45,420.48
Exp/Cntr=0.5,0.3

Type RM Length L Ch R = 1 ,206252.2,55.17,62.73,70.35
BEGIN DESCRIPTION:
18984.23  Upstream xs of Bridge 37111-0381
END DESCRIPTION:
XS GIS Cut Line= 5
  1118485.917784   672205.830778  1118388.230595   672049.473274
   1118377.34616   672029.881319   1118307.68586   671999.404929
  1118026.602535   671931.927185
#Sta/Elev= 30
       0  1089.7    24.1  1088.6    33.4    1089    55.4    1087    69.1  1084.7
   101.8  1083.2   138.8  1083.3   171.2  1082.3   193.3  1082.8   206.8  1080.1
   213.9  1077.9   218.7  1074.5   220.7  1071.3   224.7  1070.2   242.7  1071.5
   249.7    1074   256.7  1075.4   258.7  1080.2   262.5  1081.9     276  1083.1
   301.6  1088.9     321    1090   344.8  1093.1   368.4  1094.8   417.3  1093.4
   469.2  1093.7   534.1  1089.9   558.2  1097.8   567.8  1102.5   571.9    1103
#Mann= 3 , 0 , 0
       0     .13       0   218.7    .045       0   256.7     .13       0
#XS Ineff= 2 , 0
       0   195.4    1082  272.13       0    1082
Permanent Ineff=
       F       F
Bank Sta=218.7,256.7
Exp/Cntr=0.5,0.3

Type RM Length L Ch R = 3 ,206224.7,,,
BEGIN DESCRIPTION:
18956.64  Bridge : 37111-0381
END DESCRIPTION:
Bridge Culvert--1,0,-1,-1, 0
Deck Dist Width WeirC Skew NumUp NumDn MinLoCord MaxHiCord MaxSubmerge Is_Ogee
20.6,14,2.6,0, 89, 88, , , 0.95, 0, 0,0,,
      .2     1.2     8.1    16.3    17.4    28.3    29.2    30.5    39.7    50.7
      53    57.6    62.9    68.5    75.2    76.8    85.7      88    97.5   101.4
   109.4   116.7   158.1   166.7   211.7   211.7   253.7   253.7   268.6   285.3
   290.8   292.7   296.3     301   306.4   311.3   318.3     322     332   335.9
   337.6   343.9   346.3   347.1   352.6   352.7   355.1     356   356.6   364.4
   366.7   374.9   378.8   383.5     388   392.6   398.6   407.1   407.7   408.3
   408.9     422   427.2   437.1   438.9   446.3   448.3   454.7   459.1   467.4
   468.2   468.7   469.1     485   490.9   500.6   502.4   505.2     513   517.6
   526.8   531.6   540.3   543.2   544.2   546.7   554.6   557.5     571
  1087.5  1087.5  1087.3  1087.9  1087.8  1087.5  1087.5  1087.4  1087.6  1085.7
    1085  1084.8  1084.6  1084.2  1083.9  1083.8  1083.5  1083.4  1083.1    1083
  1082.7  1082.3  1082.4  1082.5  1083.5  1083.5  1083.5  1083.5  1083.5  1083.5
  1083.7  1084.2  1085.2  1085.7  1086.2  1085.9  1086.7  1087.8  1088.6  1088.8
    1089  1090.7    1091  1091.1  1091.2  1091.2    1091  1091.1  1091.1  1091.1
    1091  1091.1  1091.3  1091.4  1091.6  1091.8    1092  1092.8  1092.8  1092.8
  1092.8  1091.1  1091.6  1091.7  1091.7  1091.6  1091.3    1091  1091.1    1091
  1090.9  1090.9  1090.9  1090.1  1090.2  1090.3  1090.2  1090.3  1091.1  1090.9
  1090.3  1090.8    1094  1094.8  1095.2  1095.8  1097.2  1098.1  1102.2
                                                                                
                                                                                
                                          1080.2  1080.2
                                                                                
                                                                                
                                                                                
                                                                                
                                                                                
                                                                        
   -11.2   -10.3    -3.3     4.9       6    16.9    17.7    19.1    28.3    39.3
    41.6    46.2    51.4    57.1    63.8    65.4    74.3    76.6    86.1   121.3
   160.7     190     190     232     232   257.2   264.9   267.6   273.8   279.4
   281.3   284.9   289.6     295   299.9   306.8   310.5   320.6   324.5   326.2
   332.5   334.9   335.6   341.1   341.3   343.7   344.5   345.2     353   355.3
   363.4   367.3     372   376.5   381.1   387.1   395.7   396.3   396.9   397.4
   410.5   415.8   425.7   427.5   434.9   436.9   443.3   447.6     456   456.8
   457.3   457.7   473.5   479.4   489.2     491   493.7   501.6   506.1   515.4
   520.2   528.9   531.8   532.8   535.3   543.1   546.1   559.6
  1087.5  1087.5  1087.3  1087.9  1087.8  1087.5  1087.5  1087.4  1087.6  1085.7
    1085  1084.8  1084.6  1084.2  1083.9  1083.8  1083.5  1083.4  1083.1    1083
    1083  1083.5  1083.5  1083.5  1083.5  1083.5  1083.1  1083.2  1083.5  1083.7
  1084.2  1085.2  1085.7  1086.2  1085.9  1086.7  1087.8  1088.6  1088.8    1089
  1090.7    1091  1091.1  1091.2  1091.2    1091  1091.1  1091.1  1091.1    1091
  1091.1  1091.3  1091.4  1091.6  1091.8    1092  1092.8  1092.8  1092.8  1092.8
  1091.1  1091.6  1091.7  1091.7  1091.6  1091.3    1091  1091.1    1091  1090.9
  1090.9  1090.9  1090.1  1090.2  1090.3  1090.2  1090.3  1091.1  1090.9  1090.3
  1090.8    1094  1094.8  1095.2  1095.8  1097.2  1098.1  1102.2
                                                                                
                                                                                
                  1080.2  1080.2
                                                                                
                                                                                
                                                                                
                                                                                
                                                                                
                                                                
BR Coef=-1 , 1 , 0 ,, 0 ,,,0.8,0,1.2,0,
WSPro=,,,, 1 ,,,, 0 ,,,, 0 ,,,,-1 ,-1 ,-1 , 0 , 0 , 0 , 0 , 0
BC Design=,, 0 ,, 0 ,,,,,,

Type RM Length L Ch R = 1 ,206189.5,124.03,107.23,90.29
BEGIN DESCRIPTION:
18921.51  Down stream xs of Bridge 37111-0381
END DESCRIPTION:
XS GIS Cut Line= 4
  1118507.959239   672119.133619  1118436.122026   672005.935581
  1118335.985336   671931.921543  1118051.885926   671856.076966
#Sta/Elev= 30
       0  1086.1    22.5  1085.1    34.8    1086      84    1082   126.3  1082.1
   136.7  1081.3   149.2  1081.9   163.4  1077.7   183.6  1077.4  187.641076.491
  193.61  1073.7     203  1070.2     221  1071.5     228    1074     235  1075.4
     237  1080.2   271.3  1081.7     281  1081.3   291.6  1083.2   300.8  1082.9
   311.4  1084.3   333.3  1085.7   406.6  1087.6   412.6  1086.8   470.4  1088.1
   495.7  1089.8     506  1089.8   517.1  1088.7   531.9  1095.5   552.6  1101.6
#Mann= 3 , 0 , 0
       0     .13       0  193.61    .045       0     228     .13       0
#XS Ineff= 2 , 0
       0  172.03    1080  260.14       0 1082.12
Permanent Ineff=
       F       F
Bank Sta=193.61,228
Exp/Cntr=0.5,0.3

Type RM Length L Ch R = 1 ,206082.3,194.3,182.86,171.36
BEGIN DESCRIPTION:
18814.28
END DESCRIPTION:
XS GIS Cut Line= 6
  1118662.901658    672214.25856  1118561.768003   672129.980559
  1118494.345567   672024.633013  1118481.703893   671864.504748
  1118279.436628   671843.435248  1118056.099817   671805.510138
#Sta/Elev= 30
       0 1091.27   15.29 1091.36   24.65 1089.33    43.5 1088.97   97.45  1090.9
   119.7 1088.23  129.64 1088.27  140.17  1086.5  185.14 1086.25  207.33 1084.92
  299.42 1082.81  350.14 1083.14  375.11 1084.45  391.87 1083.62  427.74 1085.93
  448.84 1083.71  468.71 1083.25   480.5  1077.6  501.62 1069.27  507.11 1068.97
  513.12 1069.18  530.52 1077.97  591.22 1080.73  628.25 1085.46   732.5 1084.44
  793.14 1088.78   810.6 1087.24  822.04 1090.05  839.12 1097.53  847.24  1099.7
#Mann= 3 , 0 , 0
       0     .13       0   480.5    .045       0  530.52     .13       0
Bank Sta=480.5,530.52
Exp/Cntr=0.3,0.1

Type RM Length L Ch R = 1 ,205899.4,350,354.18,360
BEGIN DESCRIPTION:
18631.41
END DESCRIPTION:
XS GIS Cut Line= 4
  1118938.982387   671476.680559  1118438.298939   671656.273505
  1118304.964752    671694.36898  1117613.803924   671675.321265
#Sta/Elev= 30
       0 1157.85   16.04 1156.58   34.03 1146.73   82.05 1112.19   118.1 1100.95
  143.48 1101.32  192.67 1094.47  304.65 1090.08   361.5 1089.93  414.86 1096.11
  436.38 1094.45  499.12  1081.4  548.78 1080.53  564.08 1071.98  577.27 1071.57
  602.82 1067.33  618.75 1072.77  633.72  1078.1  755.18 1082.95  829.55 1081.73
  851.25 1086.48  895.15 1084.98  914.28 1093.56  943.53 1099.97  966.41  1100.4
  999.25 1119.82 1078.83 1145.43 1218.48 1184.52 1289.11 1193.75 1362.01  1193.2
#Mann= 3 , 0 , 0
       0     .13       0  577.27    .045       0  618.75     .13       0
Bank Sta=577.27,618.75
Exp/Cntr=0.3,0.1

Type RM Length L Ch R = 1 ,205545.2,579.09,580.63,581.12
BEGIN DESCRIPTION:
18277.23
END DESCRIPTION:
XS GIS Cut Line= 3
  1118514.615611   671195.158191  1118048.210677   671508.026106
  1117599.187333   671531.201486
#Sta/Elev= 30
       0 1168.33   57.04 1147.71   83.59 1136.48   99.49 1127.99  125.79 1119.79
  170.97 1111.04  249.64  1083.5  273.62  1080.1  321.68 1078.96  344.81 1075.31
  368.78 1076.11  416.79 1074.05  430.56 1070.76  454.38 1064.47  458.78 1064.79
  466.78 1069.79  477.69 1078.44  488.05 1082.74  539.59 1081.07  554.94 1086.16
  569.34 1096.44  582.44 1098.09  599.34 1097.36  628.52 1101.23  643.05 1107.94
  727.87 1124.31  850.38 1151.67  881.99 1156.39  941.98 1161.29 1011.24 1159.61
#Mann= 3 , 0 , 0
       0     .13       0  430.56    .045       0  466.78     .13       0
#XS Ineff= 2 , 0
          365.07 1077.81
Permanent Ineff=
       F       F
Bank Sta=430.56,466.78
Exp/Cntr=0.3,0.1

Type RM Length L Ch R = 1 ,204964.6,438.2,408.54,377.84
BEGIN DESCRIPTION:
17696.59
END DESCRIPTION:
XS GIS Cut Line= 3
  1118326.315501   670746.134847  1118004.756812   670948.919564
  1117660.022744   671177.776645
#Sta/Elev= 30
       0 1169.55   47.64  1155.3   71.65 1151.53   95.23 1141.97  130.68 1108.26
  142.38 1104.75   155.2 1089.03  167.04  1085.2   174.1 1078.83  225.41 1064.85
  250.32 1059.32  258.52 1059.99  273.85 1067.99  324.47 1078.46  333.89 1077.54
  363.73 1079.41  386.35 1086.43  410.23 1086.34  432.45 1084.28   478.8 1088.39
   530.5  1084.2  542.39 1090.93   569.7 1099.32  583.28 1097.36  594.39 1090.85
   602.3 1091.86  616.48 1095.91  631.85  1113.7   699.1  1126.2  793.94 1135.42
#Mann= 3 , 0 , 0
       0     .13       0  225.41    .045       0  273.85     .13       0
Bank Sta=225.41,273.85
Exp/Cntr=0.3,0.1

Type RM Length L Ch R = 1 ,204556.1,93.13,71.22,49.32
BEGIN DESCRIPTION:
17288.05
END DESCRIPTION:
XS GIS Cut Line= 3
  1117777.676562   670408.692548  1117773.580261   670796.351346
  1117626.093714   671007.046394
#Sta/Elev= 30
       0 1148.61   45.29 1148.67   85.13 1145.26   99.85 1144.66  143.58 1137.96
  153.64    1135  167.49 1132.08  171.82 1129.57  217.82 1095.97  250.37 1065.39
  253.28  1065.1  270.33  1059.9  281.53 1056.76  295.46 1053.98  321.13 1061.02
  345.13 1065.19  368.94 1070.91  418.89  1075.2  436.15 1074.95  451.39 1070.47
  474.91 1071.87  489.94 1080.28  514.54  1090.3  530.85 1093.68  545.48 1088.56
  567.93 1089.23  577.42 1096.08  608.84 1123.71  623.85 1127.68  644.87 1131.51
#Mann= 3 , 0 , 0
       0     .13       0  270.33    .045       0  321.13     .13       0
Bank Sta=270.33,321.13
Exp/Cntr=0.5,0.3

Type RM Length L Ch R = 1 ,204484.8,107.02,115.57,124.61
BEGIN DESCRIPTION:
17216.83  Upstream xs of Bridge 37111-0382
END DESCRIPTION:
XS GIS Cut Line= 4
  1117579.929003   670541.339718  1117676.354727   670663.623503
  1117733.131508   670744.917538  1117767.971809   670799.113547
#Sta/Elev= 30
       0  1096.4   1.697  1095.8   10.96  1095.6  12.516  1095.3   18.95  1098.6
  26.375  1100.6  27.789  1101.3   33.87  1099.9  35.002  1099.9  53.033  1093.9
  56.498  1090.6  65.832  1083.8  78.135  1076.7  82.873  1076.1 104.652  1065.9
 108.824  1065.1 115.471  1063.2 118.087  1054.8 136.472  1052.7 142.128  1054.2
 159.099  1055.6 163.412  1060.9 167.443  1061.4 176.777  1063.3 180.242  1063.4
 193.182  1068.7 206.404  1070.4 208.314    1070 214.253  1070.7 225.779  1072.8
#Mann= 3 , 0 , 0
       0     .13       0 118.087    .044       0 159.099     .13       0
#XS Ineff= 2 , 0
       0  112.64 1064.74  164.59       0 1064.85
Permanent Ineff=
       F       F
Bank Sta=118.087,159.099
Skew Angle= 45
Exp/Cntr=0.5,0.3

Type RM Length L Ch R = 3 ,204413.7,,,
BEGIN DESCRIPTION:
17145.72  Bridge : 37111-0382
END DESCRIPTION:
Bridge Culvert--1,0,-1,-1, 0
Deck Dist Width WeirC Skew NumUp NumDn MinLoCord MaxHiCord MaxSubmerge Is_Ogee
61.1,20,2.6,45, 30, 26, 1064.3, , 0.95, 0, 0,0,,
  21.779  21.991  33.517  43.275  52.962  57.134  66.609  76.509  81.742  88.105
  90.085  97.298  104.51 108.399 116.673 116.673 160.513 160.513 172.817 177.555
 179.888 180.666 190.777 195.091 210.152 213.051 224.931 226.628 233.557 234.123
  1065.6  1065.6  1065.3  1064.9  1064.6  1064.4  1064.3  1064.6  1064.8    1065
  1065.2  1065.5  1065.6  1065.7  1065.7  1065.7  1065.7  1065.7  1064.9  1064.9
  1064.9  1064.9  1066.3  1066.7  1067.9  1068.6  1071.3  1071.4  1072.7  1072.8
                                                                                
                                          1063.6  1063.6
                                                                                
  -3.889  -3.677    7.92  17.607  27.365  31.537  41.012  49.215  57.134  64.488
  71.701  82.731  88.388  88.388 132.229 132.229 147.149 151.957 154.291 154.998
  162.21 169.423 173.736 199.263 207.889 208.526
  1065.6  1065.6  1065.3  1064.9  1064.6  1064.4  1064.3  1064.7  1064.9  1065.2
  1065.5  1065.7  1065.7  1065.7  1065.7  1065.7  1064.9  1064.9  1064.9  1064.9
  1066.4  1066.7  1068.1  1071.3  1072.7  1072.8
                                                                                
                          1063.6  1063.6
                                                
Pier Skew= 45
Pier Skew, UpSta & Num, DnSta & Num=  ,127.986, 2 ,99.702, 2 , 0 , 0 , 0 ,,
       2       2
  1052.7  1064.1
       2       2
  1052.7  1064.1
Pier Skew, UpSta & Num, DnSta & Num=  ,149.2, 2 ,120.915, 2 , 0 , 0 , 0 ,,
       2       2
  1053.7  1064.1
       2       2
  1053.7  1064.1
BR Coef=-1 , 1 , 0 ,, 0 ,,,0.8,0,1,0,
WSPro=,,,, 1 ,,,, 0 ,,,, 0 ,,,,-1 ,-1 ,-1 , 0 , 0 , 0 , 0 , 0
BC Design=,, 0 ,, 0 ,,,,,,

Type RM Length L Ch R = 1 ,204369.3,159.98,181.46,202.46
BEGIN DESCRIPTION:
17101.25  Down stream xs of Bridge 37111-0382
END DESCRIPTION:
XS GIS Cut Line= 4
   1117466.15363   670587.692654  1117573.124255   670652.010069
  1117613.126057   670753.950199  1117638.933697   670817.178869
#Sta/Elev= 30
       0  1063.4   9.899  1064.5  12.233  1065.6  21.708  1065.7  40.234  1062.9
  45.184  1063.3  52.962  1062.4  55.013  1061.8  57.276  1062.1  79.125  1060.1
  88.247  1056.9  89.803  1054.8  97.581  1053.7  99.702  1053.7 108.187  1052.7
 113.844  1054.2 130.815  1055.6  133.29  1059.5 138.027  1062.8 145.452  1064.1
  147.29  1064.6 149.129  1064.3 159.311  1064.2 165.675  1064.4 183.353  1066.4
 185.969  1066.6 189.363  1066.5 195.798  1070.5 205.627  1072.6 213.971    1075
#Mann= 3 , 0 , 0
       0     .13       0  89.803    .044       0 130.815     .13       0
#XS Ineff= 2 , 0
       0   77.67  1062.5  136.61       0  1062.5
Permanent Ineff=
       F       F
Bank Sta=89.803,130.815
Skew Angle= 45
Exp/Cntr=0.5,0.3

Type RM Length L Ch R = 1 ,204187.8,531.94,569.26,605.76
BEGIN DESCRIPTION:
16919.79
END DESCRIPTION:
XS GIS Cut Line= 3
  1117773.415626   670321.343155  1117434.670369   670572.738973
  1117328.146695   670939.180383
#Sta/Elev= 30
       0 1144.61  113.36 1140.29  165.71 1133.93  179.23 1131.34  196.83 1124.87
  216.16 1120.47  231.38 1114.04  268.97 1102.74  301.02 1090.09  323.36 1072.21
  336.05 1064.83  358.55 1065.05  371.38 1066.62  391.26 1063.13  409.36 1064.72
  444.93 1059.59  462.96 1059.76  482.08 1053.75  507.15 1051.75  519.69 1052.75
  525.71 1055.97  532.23 1059.55  601.58 1068.62   617.2 1076.17  628.09 1080.34
  657.25 1086.17  751.21 1147.52  776.12 1167.43  786.71 1171.96  803.45 1174.85
#Mann= 3 , 0 , 0
       0     .13       0  482.08    .044       0  525.71     .13       0
Bank Sta=482.08,525.71
Exp/Cntr=0.3,0.1

Type RM Length L Ch R = 1 ,203618.5,345.27,368.54,391.23
BEGIN DESCRIPTION:
16350.53
END DESCRIPTION:
XS GIS Cut Line= 4
  1117979.732058   670238.612178  1117286.281302   670266.130056
  1117005.598815   670282.640801  1116631.355559   670755.948483
#Sta/Elev= 30
       0 1164.65  206.19 1137.57  286.11 1122.88  378.75 1099.52  507.84 1058.93
  584.67 1054.12  631.29 1056.98  665.63 1053.05   728.8 1053.37  742.46 1047.83
  767.76 1045.71  793.92 1048.88  883.12 1053.53  996.34 1052.55 1023.16 1055.77
 1055.62 1067.53 1083.93 1072.41 1126.82 1055.25 1147.73 1058.55 1189.88  1056.9
 1243.13 1059.89 1273.92 1068.45 1304.05 1086.52 1317.63 1099.14 1351.25 1111.64
 1401.17  1116.6 1430.84 1113.39 1462.34 1086.87 1500.66 1069.75 1578.55 1067.83
#Mann= 3 , 0 , 0
       0     .13       0  742.46    .044       0  793.92     .13       0
#XS Ineff= 2 , 0
           631.5 1058.28
Permanent Ineff=
       F       F
Bank Sta=742.46,793.92
Exp/Cntr=0.3,0.1

Type RM Length L Ch R = 1 ,203250.0,1199.09,1213.17,1226.85
BEGIN DESCRIPTION:
15982
END DESCRIPTION:
XS GIS Cut Line= 3
  1118056.099817   670208.441515  1117584.142894   670183.158079
  1116782.004923   669519.670392
#Sta/Elev= 30
       0  1171.2   63.42 1166.03  151.92 1153.65  237.56 1137.57  297.29 1123.26
  311.44 1122.61   372.5 1108.25  437.01 1089.23  511.64 1058.57  558.08 1051.44
  613.12  1049.8  660.57 1052.99  687.12 1049.52  827.12 1050.18  859.24 1048.98
  879.21 1044.05  901.93 1040.58  920.83 1044.94 1045.52 1071.18 1073.76 1084.13
 1121.86  1100.9 1143.28 1103.41 1164.86 1098.72 1185.42  1103.1 1336.48 1109.66
 1409.75 1118.96 1457.38 1122.01 1492.76 1130.83 1502.32 1129.37 1513.61 1133.13
#Mann= 3 , 0 , 0
       0     .13       0  879.21    .044       0  920.83     .13       0
#XS Ineff= 2 , 0
          660.29 1054.79
Permanent Ineff=
       F       F
Bank Sta=879.21,920.83
Exp/Cntr=0.3,0.1

Type RM Length L Ch R = 1 ,202036.8,601.49,581.57,560.65
BEGIN DESCRIPTION:
14768.82
END DESCRIPTION:
XS GIS Cut Line= 4
  1118659.782466   669777.021615  1118261.606665    669281.84551
  1118211.240857   669169.921511  1117732.070572   668772.876792
#Sta/Elev= 30
       0 1161.64   66.94 1146.99  110.73 1134.35  151.72 1117.12  164.95 1116.75
   185.1 1110.14  211.28 1120.22  245.82 1118.44  341.47 1103.33  406.93 1088.35
   417.1 1089.86  480.53 1049.53  492.99 1046.57  512.26 1046.73  531.73 1041.91
  673.58 1040.51  699.73 1038.46  725.88 1041.68  939.79 1046.97 1041.96 1053.47
 1110.75 1096.06 1120.25 1096.91 1154.71  1093.6  1188.1 1073.35 1241.58 1072.91
 1255.11 1076.07 1277.22 1091.06 1287.76 1095.15 1324.27 1104.01 1380.44 1113.15
#Mann= 3 , 0 , 0
       0     .13       0  673.58    .044       0  725.88     .09       0
Bank Sta=673.58,725.88
Exp/Cntr=0.3,0.1

Type RM Length L Ch R = 1 ,201455.3,893.66,879.31,865.16
BEGIN DESCRIPTION:
14187.25
END DESCRIPTION:
XS GIS Cut Line= 3
  1119197.629461   669151.044472  1118592.590856   668834.604727
  1117967.760744   668557.703396
#Sta/Elev= 30
       0 1120.82   15.98 1131.79   39.15 1134.25   56.08 1130.02   94.09 1100.75
  107.81 1092.64  125.85 1086.77  218.92 1078.35   241.5 1080.16  268.08 1077.27
  321.26 1064.46  462.31  1045.7  523.74 1042.03  570.95 1042.96  592.49 1038.49
     635 1036.92  661.57 1034.84  688.07 1038.26  830.24 1042.55  907.12 1040.97
  979.75  1048.4 1049.19 1048.55 1059.09 1052.42  1080.5 1070.66 1143.18 1098.22
 1160.27 1098.84 1190.59 1094.78 1228.66 1124.75 1297.48 1145.98 1366.23 1161.03
#Mann= 3 , 0 , 0
       0      .1       0     635    .044       0  688.07      .1       0
Bank Sta=635,688.07
Exp/Cntr=0.3,0.1

Type RM Length L Ch R = 1 ,200576.0,1338.56,1364.24,1382.4
BEGIN DESCRIPTION:
13307.95
END DESCRIPTION:
XS GIS Cut Line= 3
  1119661.253936   668276.133227  1119144.407273   668081.802147
  1118287.602974   668081.802147
#Sta/Elev= 30
       0 1166.99  238.18 1120.24  371.33 1116.13  431.25 1110.74  572.54 1075.47
  600.53 1058.97  617.77 1039.26  629.49 1035.13  667.26 1036.71  710.66  1033.6
   718.7 1030.54  745.35 1028.44  758.59 1029.41  771.84  1034.3  932.23  1034.4
  979.35 1046.16  988.38 1045.91 1002.76 1052.48 1010.88 1053.24 1058.54 1083.24
 1082.96 1103.42 1118.45    1116 1148.38 1117.29 1161.79 1122.37 1194.75 1121.31
 1213.85 1116.63 1333.56 1112.05 1346.12 1116.83  1403.3 1172.17 1408.98 1173.14
#Mann= 3 , 0 , 0
       0     .09       0   718.7    .044       0  771.84     .07       0
Bank Sta=718.7,771.84
Exp/Cntr=0.3,0.1

Type RM Length L Ch R = 1 ,199211.7,1230.6,1206.6,1180.67
BEGIN DESCRIPTION:
11943.71
END DESCRIPTION:
XS GIS Cut Line= 3
  1120181.163063   667762.002297  1119528.251374   667018.586527
  1118917.077581   666588.700724
#Sta/Elev= 30
       0 1116.28    3.76 1116.34    21.7 1105.21   40.66 1087.38   77.55  1069.3
  135.22 1079.59  152.14 1090.13   245.6 1093.21  466.21  1063.1  562.88    1046
   583.3 1037.49  689.44 1023.34  897.44 1025.89  914.75 1030.55  963.07 1025.65
  989.42 1022.83 1015.85 1026.66    1107 1037.98 1164.75 1092.27 1204.25 1105.57
 1300.41 1126.82 1358.91 1151.42 1459.87 1151.85 1580.43 1144.65 1615.52 1173.79
 1621.62 1175.75 1628.68 1185.59 1644.89 1200.94  1683.3 1219.53 1736.64 1227.16
#Mann= 3 , 0 , 0
       0     .09       0  963.07    .044       0 1015.85     .09       0
Bank Sta=963.07,1015.85
Exp/Cntr=0.3,0.1

Type RM Length L Ch R = 1 ,198005.1,806.22,793.4,774.51
BEGIN DESCRIPTION:
10737.11
END DESCRIPTION:
XS GIS Cut Line= 4
  1120807.777424   665560.508299  1119780.125374   665995.814595
  1119657.382377   666011.395722   1119088.50569   666331.652252
#Sta/Elev= 30
       0  1186.8  110.25 1154.71  181.77 1128.84   200.7 1123.84  219.96 1124.33
  230.99 1118.69  247.46 1117.89  320.51 1096.57  343.76  1094.5  375.81 1085.64
  395.71 1075.14  417.89 1069.73  437.22 1057.01  467.17 1044.42  732.37 1026.53
 1008.73  1021.2 1122.38 1022.14 1154.26 1016.72 1180.75 1014.57 1207.18 1021.05
 1369.35 1022.03 1395.31 1028.86 1432.14 1031.98 1467.33 1057.85 1497.11 1071.84
  1609.3 1114.27 1652.45 1128.22 1762.72  1151.1 1821.01 1150.13  1892.6 1142.98
#Mann= 3 , 0 , 0
       0     .12       0 1154.26    .043       0 1207.18     .14       0
#XS Ineff= 2 , 0
          950.41 1026.37
Permanent Ineff=
       F       F
Bank Sta=1154.26,1207.18
Exp/Cntr=0.3,0.1

Type RM Length L Ch R = 1 ,197211.7,1005.19,1000,998.18
BEGIN DESCRIPTION:
9943.711
END DESCRIPTION:
XS GIS Cut Line= 3
  1119849.134017   665044.200766  1119257.644003   665421.708349
   1118746.42063   665880.866427
#Sta/Elev= 30
       0 1128.29   41.55 1091.71  124.79 1087.59  164.78 1069.03  234.37 1027.88
  270.88 1023.85   456.3 1019.51  648.65 1017.68     661 1019.69  674.53 1017.94
   701.7 1012.12  731.12 1018.12  784.93 1019.77  845.11 1017.18  867.82 1022.97
  925.02 1019.43  960.55 1021.35  978.08 1026.13  989.41 1033.01 1007.68 1049.08
 1022.17 1057.06 1145.25 1094.42 1200.76 1107.45 1230.15  1110.9 1255.61 1118.29
 1294.52 1119.22 1307.37 1113.94 1319.44 1111.74 1351.59  1122.5 1388.84 1128.48
#Mann= 3 , 0 , 0
       0     .14       0  674.53    .043       0  731.12     .14       0
#XS Ineff= 2 , 0
                          869.93         1027.95
Permanent Ineff=
       F       F
Bank Sta=674.53,731.12
Exp/Cntr=0.3,0.1

Type RM Length L Ch R = 1 ,196211.7,950.58,971.91,992.08
BEGIN DESCRIPTION:
8943.711
END DESCRIPTION:
XS GIS Cut Line= 3
  1119277.338001   664189.379115  1118783.467075   664650.074399
  1118106.314362   665241.363749
#Sta/Elev= 30
       0 1075.34   31.24 1060.91   98.13 1046.89  117.81 1039.65  123.01 1034.43
  170.72 1028.09  306.86 1019.65  385.33 1019.25  431.39 1014.21  619.36  1015.7
  652.27 1011.24  675.39 1008.62  692.37 1009.63  705.62 1014.28  850.39 1013.15
  880.27 1019.41  909.32 1013.07 1063.96 1022.65 1106.26 1034.45 1155.53 1057.07
 1187.88 1075.94 1240.94 1078.27    1283 1112.73 1362.28 1131.41 1447.01 1133.54
 1482.01 1146.13 1492.72 1153.22 1515.16 1155.67 1529.87 1165.23 1574.36 1178.84
#Mann= 3 , 0 , 0
       0     .14       0  652.27    .043       0  705.62     .14       0
#XS Ineff= 2 , 0
                          879.12         1025.49
Permanent Ineff=
       F       F
Bank Sta=652.27,705.62
Exp/Cntr=0.3,0.1

Type RM Length L Ch R = 1 ,195239.8,1367.68,1351.11,1330.02
BEGIN DESCRIPTION:
7971.796
END DESCRIPTION:
XS GIS Cut Line= 3
   1118960.63833   663641.749847  1118423.803671   663901.779132
  1117407.359995   663948.023051
#Sta/Elev= 30
       0 1068.74   30.49  1057.2   91.81 1045.53  126.16 1025.34  171.04 1028.03
   242.5 1012.34  483.25  1015.6  561.51 1010.26  684.62 1009.42  712.79 1007.41
  740.98 1010.12  896.02 1011.92  905.28 1016.62  918.11 1017.11  944.29  1012.6
 1041.87  1015.3 1083.84  1020.8 1116.18 1040.66 1129.51 1042.91 1160.35 1043.33
 1196.76 1028.66 1248.05 1033.73  1289.5 1043.27 1323.64  1059.1 1350.18 1059.94
 1367.11 1068.98 1444.66 1078.24 1469.51 1086.61 1525.78 1093.79 1613.99 1124.52
#Mann= 3 , 0 , 0
       0     .14       0  684.62    .043       0  740.98     .14       0
#XS Ineff= 2 , 0
                          917.08         1021.26
Permanent Ineff=
       F       F
Bank Sta=684.62,740.98
Exp/Cntr=0.3,0.1

Type RM Length L Ch R = 1 ,193888.7,677.31,676.98,677.47
BEGIN DESCRIPTION:
6620.689
END DESCRIPTION:
XS GIS Cut Line= 3
  1118277.012494    662575.45004  1117664.130906   663062.612306
  1117256.038894   663643.771454
#Sta/Elev= 30
       0 1151.38  127.36 1095.95  158.74 1074.07  184.35 1062.95  219.83 1057.91
  290.65 1037.14  328.81  1039.9  364.05 1035.86  404.23 1024.13  431.14 1005.53
  469.71  999.81  497.59  997.68  525.99 1004.69  584.74 1018.21  605.99  1018.6
  641.83 1039.24  700.66 1063.64  748.81 1076.34  779.93 1079.68  824.27 1073.23
  872.99 1073.95  889.88 1072.54  910.99 1062.92  924.51 1064.69  988.51 1085.07
 1066.27 1094.38 1252.61 1152.55 1361.03 1179.59 1432.14 1195.11 1493.04 1202.19
#Mann= 3 , 0 , 0
       0     .14       0  469.71    .043       0  525.99     .14       0
Bank Sta=469.71,525.99
Exp/Cntr=0.3,0.1

Type RM Length L Ch R = 1 ,193211.7,767.99,774.75,780.53
BEGIN DESCRIPTION:
5943.711
END DESCRIPTION:
XS GIS Cut Line= 3
  1118100.826921   661860.023888  1117572.921636   662291.666174
  1117028.589302   662708.905106
#Sta/Elev= 30
       0 1247.16   33.34 1217.94   92.24 1180.06  121.69 1164.12   181.2 1139.41
  217.36  1117.8  249.27 1103.52  331.51 1080.28  401.04  1065.9  452.49 1048.86
  471.55  1053.6  486.19 1052.56  509.93 1038.71   578.2 1017.24  592.42 1008.73
  627.89  1007.9  653.59 1001.83  681.94  994.71  710.02 1002.91  743.85 1017.11
  772.74 1019.07   820.2 1048.83  898.82 1082.68  956.48 1083.28  968.75 1087.32
 1088.51 1101.96 1121.33 1102.98 1220.21 1154.28 1274.91 1174.89 1367.76 1230.29
#Mann= 3 , 0 , 0
       0     .14       0  653.59    .043       0  710.02     .14       0
Bank Sta=653.59,710.02
Exp/Cntr=0.3,0.1

Type RM Length L Ch R = 1 ,192437.0,169.72,192.18,214.64
BEGIN DESCRIPTION:
5168.957
END DESCRIPTION:
XS GIS Cut Line= 2
   1117611.30578   661412.442417  1116659.186849   661885.750099
#Sta/Elev= 30
       0 1131.77   71.67 1104.05  142.55 1070.03  169.68 1062.89  189.45 1048.57
  244.25 1042.87   293.6 1015.38  332.03 1000.78  441.77  993.34  469.67  985.55
  480.36  986.86  498.42  995.19  509.32   995.6  530.67 1007.14  549.13 1006.43
  594.69 1023.91   648.2 1050.58  675.56 1056.94  724.09 1055.53  735.96 1058.32
  758.07 1079.89  843.65 1111.35  925.75 1146.19  977.05 1162.57  998.84 1166.32
  1018.2 1165.23 1031.71 1159.69 1043.35 1148.58 1056.26 1141.32 1063.27 1145.18
#Mann= 3 , 0 , 0
       0     .14       0  441.77    .042       0  498.42     .14       0
Bank Sta=441.77,498.42
Exp/Cntr=0.5,0.3

Type RM Length L Ch R = 1 ,192244.8,141.57,148.25,156.86
BEGIN DESCRIPTION:
4976.778  Upstream xs of Bridge 37111-0395
END DESCRIPTION:
XS GIS Cut Line= 5
  1117415.514391   661487.463949  1117235.682178   661580.976696
  1117165.202565   661465.909559  1117016.605993   661443.895248
  1116577.496373    661670.89278
#Sta/Elev= 30
       0  1046.7  26.517  1043.1  38.749  1034.6  67.175  1009.2  84.499  1000.3
  117.45   999.2 133.077   995.9 233.416   996.8 263.397   992.7 266.438   986.2
 279.873   984.6 304.622   987.3   312.4   987.8 315.087   993.6 345.351   994.2
  357.23   999.7 383.464  1006.5 391.454  1004.8 415.991  1008.8 429.426  1017.8
 442.366  1022.9 460.185  1039.5 473.832  1046.6 525.239  1045.4 571.696  1062.1
  592.98  1062.6 617.799    1058 659.306  1063.1 674.721  1069.7  694.52    1072
#Mann= 3 , 0 , 0
       0     .14       0 266.438    .042       0 304.622     .14       0
#XS Ineff= 2 , 0
       0 220.971   996.1 357.867       0   996.1
Permanent Ineff=
       F       F
Bank Sta=266.438,304.622
Skew Angle= 45
Exp/Cntr=0.5,0.3

Type RM Length L Ch R = 3 ,192170.5,,,
BEGIN DESCRIPTION:
4902.502  Bridge : 37111-0395
END DESCRIPTION:
Bridge Culvert--1,0,-1,-1, 0
Deck Dist Width WeirC Skew NumUp NumDn MinLoCord MaxHiCord MaxSubmerge Is_Ogee
63.3,22,2.6,45, 150, 127, 996.2, , 0.95, 0, 0,0,,
  14.708  17.041  22.415  25.385  33.093  33.588    33.8  42.426  47.235   50.77
  55.296  59.821  69.014  69.862  71.701  76.792  79.055  88.388  93.338 101.046
   105.5 111.864 114.056 116.602  120.42 123.107 130.956 131.734 132.088 138.522
 140.714  147.22 148.917 154.715 155.281 155.422 155.846 164.119 166.736 168.433
  170.13 172.534 177.484 182.716 183.282 183.848  190.99 192.333 197.566 204.425
 205.556 206.475  210.93 212.132 216.728 218.425 222.385 224.294 225.779 232.072
 236.103 238.578  242.82  246.71 251.518 252.225 253.003 265.731 265.731 313.107
 313.107 326.683 331.492 344.856 350.089 357.301  363.17 364.372 370.736 371.231
 371.585 377.312 383.888  385.09 385.939 390.747 394.283 401.707 404.889  415.92
 420.092 426.668 427.517 428.365 446.326 449.508 454.175 457.074 461.034 469.802
 476.802  483.59 493.207  495.54 500.632 505.086 515.481 526.724  527.36 527.997
 552.958 561.726  564.13 573.605  580.11  584.07 585.343 586.687 596.515  602.95
 607.193 609.102 616.809 617.446 632.295 633.285 634.133 636.538 640.639 642.831
  649.76 657.609 659.094 660.438 667.085 674.792 675.358  676.63 687.237 692.399
 699.399 701.026 703.713 713.683 720.825 721.885 731.785 733.765 740.341 743.947
  1045.2  1044.8  1044.8  1044.8  1043.8  1043.8  1043.7  1038.5  1035.5  1032.6
  1029.2  1026.8  1019.7  1019.2  1018.1  1014.8  1012.9  1003.9  1001.7   999.8
   999.2   998.4   998.2   998.2   998.3   998.2   997.6   997.6   997.6   997.7
   997.5   997.5   997.4   997.3   997.3   997.3   997.3   997.8   997.9   997.7
   997.7   997.7     998   997.2   997.2   997.2   997.2   997.1     997     997
   996.9   996.9   996.9     997     997   996.9   996.7   996.6   996.6   996.8
   996.6   996.2   996.1   996.1   996.2   996.1   996.2   996.2   996.2   996.2
   996.2   997.5   997.5   998.7   998.9     999   999.3   999.4   999.3   999.3
   999.3   999.2   999.1   999.1   999.1   999.3   999.3   999.1   999.1   998.9
   998.8   998.9   998.9   998.9   997.1   996.9   996.6   996.4   996.5   996.7
     996     996   995.8   995.7   994.9   993.8   994.2   999.3   999.6   999.7
  1000.3  1000.3  1000.5  1002.2  1003.7  1004.1  1004.3  1004.3  1005.4    1008
  1009.6  1010.9  1018.7  1019.5  1031.9  1032.8  1033.4  1033.9  1034.4  1034.3
  1033.9  1034.1  1034.1  1033.6  1031.3  1024.3  1023.7  1022.9  1015.1  1015.8
    1017  1017.7  1018.9  1023.3  1026.4  1026.9  1031.6  1032.6  1036.2  1038.3
                                                                                
                                                                                
                                                                                
                                                                                
                                                                                
                                                                                
                                                                   994.2   994.2
                                                                                
                                                                                
                                                                                
                                                                                
                                                                                
                                                                                
                                                                                
                                                                                
  30.193  32.456   37.83    40.8  48.508  49.003  49.215  57.912   62.65  66.185
  70.711  75.307  84.429  85.277  87.116  92.207  94.469 103.874 108.753  116.46
 120.915 127.279 129.471 146.442 147.149 147.502 156.129 164.332  170.13 170.696
 170.837 171.261 198.131 198.697 199.333 206.404 207.748 212.981 219.839 220.971
  221.89 226.345 227.547 232.143 233.911   237.8  239.78 241.194 253.993 258.235
 262.195 266.933  267.64 268.418 281.216 281.216 328.593 328.593 342.098 352.917
 367.696 379.787 386.151 386.646     387 392.727 401.354 406.162 417.193 420.304
 425.678 431.335 435.507 442.083 443.002  443.78 448.447 461.811 464.923  469.59
 476.449 492.217 499.005 508.622 510.955 516.047 520.501 530.896 542.139 542.775
 568.372 579.545  589.02 595.596 599.485 600.758 602.172 612.001 618.365 622.607
 624.587 632.224 632.861  647.71   648.7 649.619 651.952 656.054 673.024 674.509
 675.853 682.499 690.207 690.843 692.045 702.723 707.814 714.814 716.441 719.128
 729.098  736.24 737.371   747.2  749.18 755.826 759.362
  1045.2  1044.8  1044.8  1044.8  1043.8  1043.8  1043.7  1038.5  1035.5  1032.6
  1029.2  1026.8  1019.7  1019.2  1018.1  1014.8  1012.9  1003.9  1001.7   999.8
   999.2   998.4   998.2   997.6   997.6   997.6   997.5   997.4   997.3   997.3
   997.3   997.3   997.2   997.2   997.2   997.2   997.1     997     997   996.9
   996.9   996.9     997     997   996.9   996.7   996.6   996.6   996.2   996.1
   996.1   996.2   996.1   996.2   996.2   996.2   996.2   996.2   997.5   999.2
   999.2   999.4   999.3   999.3   999.3   999.2   999.1   999.3   999.1   999.1
   999.2   998.9   998.8   998.9   998.9   998.9   997.7   997.1   996.9   996.6
   996.5     996     996   995.8   995.7   994.9   993.8   994.2   999.3   999.6
  1000.3  1000.5  1002.2  1003.7  1004.1  1004.3  1004.3  1005.4    1008  1009.6
  1010.9  1018.7  1019.5  1031.9  1032.8  1033.4  1033.9  1034.4  1034.1  1034.1
  1033.6  1031.3  1024.3  1023.7  1022.9  1015.1  1015.8    1017  1017.7  1018.9
  1023.3  1026.4  1026.9  1031.6  1032.6  1036.2  1038.3
                                                                                
                                                                                
                                                                                
                                                                                
                                                                                
                                           994.2   994.2
                                                                                
                                                                                
                                                                                
                                                                                
                                                                                
                                                                                
                                                        
Pier Skew= 45
Pier Skew, UpSta & Num, DnSta & Num=  ,289.801, 2 ,305.23, 2 , 0 , 0 , 0 ,,
       1       1
   983.6   994.7
       1       1
   983.6   994.7
BR Coef=-1 , 1 , 0 ,, 0 ,,,0.8,0,1.2,0,
WSPro=,,,, 1 ,,,, 0 ,,,, 0 ,,,,-1 ,-1 ,-1 , 0 , 0 , 0 , 0 , 0
BC Design=,, 0 ,, 0 ,,,,,,

Type RM Length L Ch R = 1 ,192096.6,265.76,246.99,226.06
BEGIN DESCRIPTION:
4828.53  Down stream xs of Bridge 37111-0395
END DESCRIPTION:
XS GIS Cut Line= 6
  1117433.497573   661206.925751  1117121.173941   661344.830867
  1116983.584503    661306.30581  1116890.023689   661185.227117
  1116847.244671   661142.186174  1116552.319866   661357.984794
#Sta/Elev= 30
       0  1094.9  22.274  1080.6  29.486  1073.3  86.126  1046.1  111.44  1040.3
 142.411  1026.3 179.959  1014.7 197.424  1005.6 241.406   995.9 278.883   991.7
 281.923   986.2 295.359   984.6 320.107   987.3 327.885   987.8 331.492   993.1
 342.452   995.1 432.042   992.6 498.369     994 517.956   997.3 539.947   993.8
 552.816   999.2 627.345  1005.8 644.104  1017.4 654.781  1028.9 667.014    1032
 690.419  1030.9 706.329  1016.6  717.36    1015 730.158    1016 751.937    1027
#Mann= 3 , 0 , 0
       0     .14       0 281.923    .042       0 320.107     .14       0
#XS Ineff= 2 , 0
       0 236.669   996.2  373.07       0   996.2
Permanent Ineff=
       F       F
Bank Sta=281.923,320.107
Skew Angle= 45
Exp/Cntr=0.5,0.3

Type RM Length L Ch R = 1 ,191849.6,915.87,905.38,894.83
BEGIN DESCRIPTION:
4581.54
END DESCRIPTION:
XS GIS Cut Line= 5
  1117336.388207   660865.244595  1116963.275143    661098.61343
  1116878.951918   661108.938699  1116559.513147   661343.598231
  1116271.781624   661577.380077
#Sta/Elev= 30
       0 1154.99   26.51 1137.62   41.44    1122   81.35 1091.55  127.28 1063.69
  159.58 1052.45   174.9 1042.24  209.08 1038.56  369.79   998.4  406.07  992.43
  456.77  990.54  484.41  984.14  513.32  992.36  603.37  997.26  639.03  994.19
  656.32  999.46  751.26  1003.6  768.63 1008.58  800.42 1029.03  817.26 1031.65
  845.55 1031.06  870.78 1017.73  894.52 1014.34 1024.79 1056.85 1099.62 1066.56
 1187.62 1094.78 1211.11 1093.82 1242.29 1085.68  1273.1 1071.92 1292.14 1058.73
#Mann= 3 , 0 , 0
       0     .14       0  456.77    .042       0  513.32     .14       0
Bank Sta=456.77,513.32
Exp/Cntr=0.3,0.1

Type RM Length L Ch R = 1 ,190944.2,724.02,722.53,720.96
BEGIN DESCRIPTION:
3676.165
END DESCRIPTION:
XS GIS Cut Line= 4
  1117163.017877   659988.402235  1116554.802373   660298.047494
  1116075.800278   660541.909698  1115293.986193    661306.30581
#Sta/Elev= 30
       0 1227.81   33.63 1215.22  105.94 1200.02   129.7 1188.08  211.53 1177.09
   281.7 1147.94  349.14 1107.26  412.89 1032.34  446.66 1029.38  508.94  991.18
  568.83  988.59  582.38  983.09  611.22  981.03  640.28  986.57  994.04  989.29
 1268.99 1008.71  1284.9 1020.74 1365.19 1046.54 1422.31 1054.61 1483.05 1055.29
 1593.91 1094.96  1726.7 1119.43  1811.5 1117.81 1898.57  1127.2    2008 1127.54
 2081.24 1117.01 2114.69 1097.45 2197.47 1114.97 2256.38 1112.73 2313.41 1140.51
#Mann= 3 , 0 , 0
       0     .14       0  582.38    .042       0  640.28      .1       0
Bank Sta=582.38,640.28
Exp/Cntr=0.3,0.1

Type RM Length L Ch R = 1 ,190221.7,1225.73,1233.28,1240.49
BEGIN DESCRIPTION:
2953.633
END DESCRIPTION:
XS GIS Cut Line= 4
  1117005.598815   659418.578693  1116493.766121   659534.153863
  1116273.623002   659660.736123  1115671.142115   659886.957478
#Sta/Elev= 30
       0  1211.4   23.12 1207.65   61.78 1195.25   97.93 1176.68  142.86 1149.01
  218.38 1113.83  291.22 1084.46  370.54 1058.76  483.45 1014.73   496.1 1015.61
  518.56 1024.34  535.47 1022.87  546.54 1016.37  588.69   983.1  594.85  980.15
  598.64  981.29  625.92   978.3  642.46   979.3  657.05  985.78  876.39  984.34
  951.39   986.4  996.91  983.89 1041.25  987.15 1079.21  985.02 1156.08  987.46
 1289.81  986.08 1327.73  989.94 1360.81 1009.86 1367.15 1011.16 1422.21 1009.87
#Mann= 3 , 0 , 0
       0     .14       0  598.64    .042       0  657.05      .1       0
Bank Sta=598.64,657.05
Exp/Cntr=0.3,0.1

Type RM Length L Ch R = 1 ,188988.4,1490.39,1507.43,1520.5
BEGIN DESCRIPTION:
1720.354
END DESCRIPTION:
XS GIS Cut Line= 3
  1116398.032747   658443.493131  1115725.091792   658674.888515
  1114958.045029   658892.232783
#Sta/Elev= 30
       0 1108.93  139.72 1046.05  223.66 1014.85  243.15 1011.19  279.03 1014.43
  320.77  997.31  360.82  992.94   393.2  983.48   509.2  982.63  528.14  973.97
  574.62  972.25  736.67  980.99   753.7  974.74  799.64  974.52  814.62  980.12
  905.99  987.85  926.55  1006.7 1003.89 1037.54  1049.3 1030.21 1069.01  1010.7
 1080.26 1006.13  1129.4 1007.35 1177.86 1053.39 1204.49 1067.91 1251.29 1070.53
 1326.35 1067.99 1375.98 1061.02 1407.71 1051.51 1432.47 1053.91 1508.86 1074.76
#Mann= 3 , 0 , 0
       0     .14       0   753.7    .042       0  799.64      .1       0
#XS Ineff= 2 , 0
          509.14  982.63
Permanent Ineff=
       F       F
Bank Sta=753.7,799.64
Exp/Cntr=0.3,0.1

Type RM Length L Ch R = 1 ,187481. ,248.45,212.92,237.36
BEGIN DESCRIPTION:
212.921
END DESCRIPTION:
XS GIS Cut Line= 3
  1116488.262554   657651.930313  1115618.697303   657442.794373
  1114705.824965   657255.587717
#Sta/Elev= 30
       0 1134.29   47.18 1138.66   94.38 1134.78  250.93 1104.76  428.09 1050.66
   479.9 1028.57  505.34 1006.63  552.34  1002.2  579.01  985.55  607.94  976.32
  663.73  972.42  687.17  967.17  716.88  964.63  731.74  965.37   746.6  970.87
  785.24  974.62 1014.83  975.65 1053.59  982.23 1176.42  976.08 1204.39  978.87
 1233.98  996.61 1251.51 1000.23 1285.02 1000.26  1323.9  979.16 1353.88  977.55
 1514.59  979.57 1566.96   989.6 1629.37  989.31 1679.97  997.74 1826.23   997.8
#Mann= 3 , 0 , 0
       0      .1       0  687.17    .042       0   746.6     .14       0
Bank Sta=687.17,746.6
Exp/Cntr=0.3,0.1
Stream Node=2ndBroadRv      ,Main            , 0 , 0 ,Upstream end
Stream Node=2ndBroadRv      ,Main            , 0 , 1 ,Downstream end

Chan Stop Cuts=-1
Use User Specified Reach Order=0
User Specified Reach Order=2ndBroadRv      ,Main
